HEC-RAS study KNAPPCK.prj: KNAPPCK

--- KNAPPCK.g01 (geometry) --- (continued)

Type RM Length L Ch R = 1 ,146263  ,335,324.6,313.1
XS GIS Cut Line= 4
2304241.32187263467315.5968640782304112.62833813 467466.42388448
2303915.15839953467576.0286083832303784.12260959467825.111087851
#Sta/Elev= 30
       0 2859.55    70.4 2835.26    89.9 2829.95   129.6 2817.52   191.4 2800.59
   198.8 2798.23   212.4 2792.06   218.3 2791.14   244.8 2791.93   264.3 2789.68
     272 2788.75   278.1 2789.54   281.1 2790.62   290.3  2791.6   322.3    2791
     336 2792.69   362.4 2791.59     386 2791.64   429.3 2793.16   468.6 2791.48
   495.3 2792.85   520.3 2791.31   538.4 2793.21     552 2793.17   628.6 2799.75
   646.9 2803.83   661.2    2806   679.7 2811.18   692.1 2813.41   705.6 2817.64
#Mann= 5 ,-1,0
       0      .1       0   264.3    .045       0   278.1      .1       0
  461.26     .06       0  571.26      .1       0
#XS Ineff= 2 , 0
                          494.87         2798.99
Permanent Ineff=
       F       F
Bank Sta=264.3,278.1
XS Rating Curve= 0 ,0
Exp/Cntr(USF)=0,0
Exp/Cntr=0.3,0.1

Type RM Length L Ch R = 1 ,145939  ,75.5,75.3,76.1
XS GIS Cut Line= 3
 2303879.0274753467190.3362153912303694.93118228 467577.35654758
2303610.60460307467739.234408883
#Sta/Elev= 30
       0 2820.75      43 2810.87    51.9 2807.86    65.2 2799.18      74 2790.73
    79.3 2787.67    96.2 2785.78   124.3 2785.42   136.72783.637   144.9 2782.89
   154.4 2783.62   158.2 2786.64   162.6 2787.19   184.4 2786.41   211.5 2787.91
   237.9 2786.34   264.5 2787.18   289.4 2786.52   343.5 2788.12   379.7 2786.56
   391.5 2787.32   401.8 2785.21   410.7 2788.38   415.1 2788.93   459.9 2787.49
   518.6 2790.41   528.3 2792.03   546.1 2797.18   584.7 2811.44   611.1 2818.09
#Mann= 5 ,-1,0
       0      .1       0   136.7    .045       0   154.4      .1       0
     380     .06       0  508.57      .1       0
#XS Ineff= 2 , 0
                             420         2797.26
Permanent Ineff=
       F       F
Bank Sta=136.7,154.4
XS Rating Curve= 0 ,0
Exp/Cntr(USF)=0,0
Exp/Cntr=0.3,0.1

Type RM Length L Ch R = 1 ,145863  ,418.2,416.2,415
XS GIS Cut Line= 3
2303801.20703434467191.672856623 2303583.3449765467597.767732433
2303557.20152956467718.027588359
#Sta/Elev= 30
       0 2820.25    10.8 2817.37    47.1 2805.68    52.1 2803.08    56.2 2800.04
    65.3 2792.19    69.8 2786.86    74.3 2783.51    81.6 2783.72    86.8  2782.7
    95.3    2782   103.7 2782.09  106.65  2782.8   114.1 2786.61   120.6 2786.82
   137.6 2786.37   342.2 2786.19   353.7  2785.2   374.1 2785.86     383 2786.88
   396.6 2787.48   414.8 2786.23   424.3 2786.72   442.2 2786.16   464.3 2787.16
   473.1 2789.81   517.5 2808.73   533.9 2814.87   550.4 2819.68   583.9 2827.27
#Mann= 5 ,-1,0
       0      .1       0    86.8    .045       0  106.65      .1       0
   120.6     .06       0   414.8      .1       0
#XS Ineff= 2 , 0
                          395.15         2794.01
Permanent Ineff=
       F       F
Bank Sta=86.8,106.65
XS Rating Curve= 0 ,0
Exp/Cntr(USF)=0,0
Exp/Cntr=0.3,0.1

Type RM Length L Ch R = 1 ,145447  ,489.8,490.4,486.8
XS GIS Cut Line= 2
2303412.41200821467035.7860229482303172.95045056467587.373335056
#Sta/Elev= 30
       0 2824.39    23.3 2804.91    45.1 2782.99    49.5 2779.87    53.8 2778.88
    62.6  2779.5    88.7 2779.56   106.2 2778.78   114.9 2779.26     1192778.666
     128 2777.78   145.4 2778.64   154.1 2779.42   175.9 2778.78     189 2779.82
   202.1 2780.08   228.3 2778.46     298 2776.72     346 2779.53   376.5 2779.34
   392.3 2780.78   407.1 2780.61   420.1 2779.29   448.2 2780.22   472.3 2782.35
   498.6  2785.7   516.1 2790.72   521.2 2792.78   564.8  2814.7   601.3 2834.72
#Mann= 5 ,-1,0
       0      .1       0     119    .045       0   145.4      .1       0
     330     .06       0     540      .1       0
#XS Ineff= 2 , 0
           88.34 2784.69   398.7         2789.35
Permanent Ineff=
       F       F
Bank Sta=119,145.4
XS Rating Curve= 0 ,0
Exp/Cntr(USF)=0,0
Exp/Cntr=0.3,0.1

Type RM Length L Ch R = 1 ,144957  ,351.3,349.5,354.9
XS GIS Cut Line= 2
2303025.31363892466961.7467429832302816.23530261 467448.65077752
#Sta/Elev= 30
       0  2794.1    53.6  2777.9    73.4 2776.75   104.3 2771.12   114.4 2770.02
   121.3 2770.15   135.12768.156   147.4 2767.84   151.7 2768.17   160.4 2771.53
   173.5 2772.64   282.3 2773.05   304.1 2770.73   308.5 2771.25   317.2 2773.94
   334.6    2774   347.6 2772.75   368.9 2773.62   382.5 2779.47   391.2 2785.24
   399.9 2792.65   404.2 2794.63   421.6 2797.63     439 2802.45   457.3 2808.47
   465.2 2812.24   478.6 2812.75   486.9 2816.08   504.4 2820.95   529.9 2833.05
#Mann= 5 ,-1,0
       0      .1       0   135.1    .045       0   151.7      .1       0
     310     .06       0     410      .1       0
#XS Ineff= 2 , 0
                          214.99          2779.2
Permanent Ineff=
       F       F
Bank Sta=135.1,151.7
XS Rating Curve= 0 ,0
Exp/Cntr(USF)=0,0
Exp/Cntr=0.3,0.1

Type RM Length L Ch R = 1 ,144607  ,344.8,334.2,320.8
XS GIS Cut Line= 2
2302723.06039257466888.8265587032302527.22997441467339.654482313
#Sta/Elev= 30
       0 2778.25    13.5 2773.11    20.7 2771.25    57.1 2767.48      92 2767.56
   108.9  2768.5   139.9 2767.03     153 2767.29   169.7 2765.59   179.2 2765.98
   187.9 2764.13   218.4 2766.22   231.5  2765.6   238.9 2764.06   244.6 2762.91
   251.8 2762.88   257.7 2762.96     262 2764.03   266.4 2767.41   275.1 2768.88
   296.9 2768.66   312.6 2765.51   358.2 2765.95   375.4 2769.11   384.2 2773.95
   414.7 2802.28   432.1 2816.47   480.1 2846.96   484.5 2848.87   491.5 2849.59
#Mann= 5 ,-1,0
       0      .1       0   238.9    .045       0     262      .1       0
     280     .06       0     390      .1       0
#XS Ineff= 2 , 0
                          281.97         2778.72
Permanent Ineff=
       F       F
Bank Sta=238.9,262
XS Rating Curve= 0 ,0
Exp/Cntr(USF)=0,0
Exp/Cntr=0.3,0.1

Type RM Length L Ch R = 1 ,144273  ,193,157.1,113.8
BEGIN DESCRIPTION:
structure xs 4
END DESCRIPTION:
XS GIS Cut Line= 3
2302400.65354212466742.0178122952302400.65354212 467007.06679054
2302341.52723159467265.999253902
#Sta/Elev= 30
       0 2781.34    31.2 2775.26    55.2 2767.76    71.2  2764.8   115.2 2763.26
   139.2 2763.32   147.2 2762.58   167.32758.542   171.2 2757.57   182.7  2757.5
   196.92758.499   203.2 2760.01   210.7 2760.56   239.2 2760.73   247.6 2761.52
   275.4 2768.58   283.6 2767.82   295.9 2764.49   332.9 2765.53   349.3 2762.36
     378 2761.02   397.5 2764.23   405.5 2764.03   423.1 2764.69   427.2 2766.63
   442.7  2778.3   484.3 2814.39     497  2823.6   517.5 2836.39   530.6 2845.79
#Mann= 5 ,-1,0
       0      .1       0   167.3    .045       0   196.9      .1       0
   210.7     .06       0   405.5      .1       0
#XS Ineff= 2 , 0
                          275.83         2781.01
Permanent Ineff=
       F       F
Bank Sta=167.3,196.9
XS Rating Curve= 0 ,0
Exp/Cntr(USF)=0,0
Exp/Cntr=0.5,0.3

Type RM Length L Ch R = 1 ,144116  ,92.5,98.3,109.4
BEGIN DESCRIPTION:
structure xs 3
END DESCRIPTION:
XS GIS Cut Line= 4
2302079.29185019466706.4400840612302107.06082775466890.853007771
2302375.18845182 466984.272578412302314.43107066 467259.82157387
#Sta/Elev= 30
       0 2775.66    67.5 2764.33    75.6 2760.15    79.6 2759.16     116 2755.77
   140.3 2756.44   176.7 2757.89   205.7 2756.56   285.1 2758.55   310.5 2756.72
     318 2755.41   358.8 2756.74   382.5  2758.8   420.6 2759.17   470.4  2761.2
   487.1 2766.98   493.9 2767.93   500.6 2767.77     514 2764.13   553.3 2765.07
   569.7 2762.06   594.2  2760.6   614.7 2761.72   630.6 2763.91   644.9 2765.35
   663.9 2775.23   676.2 2784.66   696.6 2803.19   729.4 2830.54   752.6  2846.8
#Mann= 5 ,-1,0
       0      .1       0   140.3     .06       0   310.5    .045       0
   358.8     .06       0   630.6      .1       0
#XS Ineff= 2 , 0
           254.5 2759.94   414.8          2763.5
Permanent Ineff=
       F       F
Bank Sta=310.5,358.8
XS Rating Curve= 0 ,0
Exp/Cntr(USF)=0,0
Exp/Cntr=0.5,0.3

Type RM Length L Ch R = 1 ,144018  ,228.1,268.1,306.8
BEGIN DESCRIPTION:
structure xs 2
END DESCRIPTION:
XS GIS Cut Line= 4
2302035.73207003466738.4294568972302080.55592993 466968.32886295
2302296.96842067467052.9610405422302262.71593732467257.150695705
#Sta/Elev= 30
       0 2768.55    23.2 2763.34    39.5 2756.64    59.9 2755.09   111.9 2756.47
   129.1 2755.81     178 2757.05   190.4 2759.11   210.5 2759.81   274.4 2760.47
   293.9 2760.78   319.22755.058   344.9 2754.89   350.52755.046   375.6 2757.12
   384.1 2761.25   390.3 2762.57   435.3 2763.59     479 2764.11   523.6 2760.11
   547.9 2763.83     552 2766.11   571.7 2782.63   604.7 2807.84   616.9 2815.82
   633.1 2828.82   653.4 2842.02   661.5 2848.67   665.6 2850.79   673.6  2852.1
#Mann= 7 ,-1,0
       0      .1       0   111.9     .06       0   210.5      .1       0
   274.4     .06       0   319.2    .045       0   350.5     .06       0
   435.3      .1       0
#XS Ineff= 3 ,-1
   17.08  207.42 2763.08  207.42  315.95 2758.18     354   673.6    2763
Permanent Ineff=
       F       F       F
Bank Sta=319.2,350.5
XS Rating Curve= 0 ,0
Exp/Cntr(USF)=0,0
Exp/Cntr=0.5,0.3

Type RM Length L Ch R = 1 ,143750  ,258.6,258.5,258.4
BEGIN DESCRIPTION:
structure xs 1
END DESCRIPTION:
XS GIS Cut Line= 2
2302030.31895436466743.3634455692301878.32355953 467142.13982753
#Sta/Elev= 30
       0 2767.14     6.2 2764.54    17.3 2757.32    21.7 2756.04    53.3 2754.78
    86.8 2754.75    99.1 2753.14   104.7 2753.25   111.5 2754.63   143.2 2754.95
     156 2756.84   168.9  2757.3   181.7 2756.97   190.3 2755.46     220 2754.79
   237.4 2756.07   255.82750.071   263.1  2749.1   275.9 2749.16   284.5 2750.17
   288.8 2752.25   296.9 2761.99   305.9  2774.3   324.5 2790.45   335.8 2798.97
   342.9 2802.26   387.4 2817.73     400 2824.38   409.1 2825.65   426.8 2835.33
#Mann= 5 ,-1,0
       0      .1       0   111.5     .06       0     220      .1       0
   255.8    .045       0   284.5      .1       0
#XS Ineff= 2 , 0
          167.61 2765.63
Permanent Ineff=
       F       F
Bank Sta=255.8,284.5
XS Rating Curve= 0 ,0
Exp/Cntr(USF)=0,0
Exp/Cntr=0.3,0.1

Type RM Length L Ch R = 1 ,143491  ,319.2,320.1,320.9
XS GIS Cut Line= 2
2301813.79967851  466579.98333392301627.18480944467078.723957423
#Sta/Elev= 30
       0 2768.58    14.1    2762    39.7 2754.81    61.1 2752.21    73.9 2749.39
    95.2 2750.24   103.8 2749.18   116.6 2750.19     155 2750.35   167.8 2748.75
   180.7  2748.9   197.7 2750.43   219.1 2749.59   227.6 2751.89   240.4 2752.42
   253.3 2752.07   270.3 2749.39     290 2749.79   317.3 2750.91   328.9 2746.11
   334.4 2745.63   353.4 2746.18   368.6 2752.39   381.4 2764.68   394.2 2774.62
   441.2 2798.59   458.3 2809.12   468.4 2811.33   477.7 2817.75   532.5 2848.66
#Mann= 5 ,-1,0
       0      .1       0   180.7     .06       0     290      .1       0
   328.9    .045       0   353.4      .1       0
#XS Ineff= 2 , 0
           316.1 2765.18
Permanent Ineff=
       F       F
Bank Sta=328.9,353.4
XS Rating Curve= 0 ,0
Exp/Cntr(USF)=0,0
Exp/Cntr=0.3,0.1

Type RM Length L Ch R = 1 ,143171  ,309.9,310.9,311.2
XS GIS Cut Line= 2
2301523.44598892466485.0209465192301315.05905498 466976.33349829
#Sta/Elev= 30
       0 2767.51    42.3 2755.47    57.5 2745.78    72.8 2744.58   130.5 2744.07
     145  2744.7   178.3 2742.87     200 2743.48   208.7 2745.75   219.2 2746.47
   234.8 2746.29   247.8 2743.47   256.5  2745.6   291.3 2745.82   308.7 2741.85
   325.9 2741.59   329.1 2741.84   336.2  2744.4   343.4 2745.35   369.5  2743.8
   374.8  2744.4   378.2 2746.27   395.6 2760.14   435.8 2794.73   456.4 2804.91
   465.1 2810.26   473.8 2811.54   478.1  2813.2   487.7 2819.19   533.7 2841.96
#Mann= 5 ,-1,0
       0     .12       0    72.8     .06       0   291.3      .1       0
   308.7    .045       0   329.1      .1       0
#XS Ineff= 2 , 0
          289.06 2755.53
Permanent Ineff=
       F       F
Bank Sta=308.7,329.1
XS Rating Curve= 0 ,0
Exp/Cntr(USF)=0,0
Exp/Cntr=0.3,0.1

Type RM Length L Ch R = 1 ,142860  ,351.7,352,348.9
XS GIS Cut Line= 2
 2301246.7939994466377.2306180762301016.34587828466877.033685974
#Sta/Elev= 30
       0 2741.06    26.4 2740.24   114.5 2739.74   149.6 2737.91   198.2 2738.06
   209.9 2740.02     222 2740.55   246.6 2738.91   259.8  2738.7   273.3 2739.93
   276.3 2739.67   281.8 2737.61   290.7 2736.22   294.52735.003   299.5 2734.48
   315.5 2735.06   356.7 2740.22   361.1 2743.09   374.3 2753.86   387.8 2763.78
   396.4 2768.93   405.2 2771.43     427 2775.29   436.1 2779.74   444.8 2780.24
   449.2 2781.21     458 2786.85   490.3 2802.22   522.1 2816.23   550.4 2830.18
#Mann= 4 ,-1,0
       0      .1       0     190     .06       0   294.5    .045       0
   315.5      .1       0
#XS Ineff= 2 , 0
          225.13 2749.85
Permanent Ineff=
       F       F
Bank Sta=294.5,315.5
XS Rating Curve= 0 ,0
Exp/Cntr(USF)=0,0
Exp/Cntr=0.3,0.1

Type RM Length L Ch R = 1 ,142508  ,366.3,359.4,344.5
XS GIS Cut Line= 2
2300933.57202176466279.417792572 2300720.5338084466741.826317693
#Sta/Elev= 30
       0 2734.95    32.8 2735.56    41.6 2735.31    62.7 2733.78    89.8 2733.63
    98.9 2734.09   138.5 2733.11   175.4 2733.47   201.4 2734.62   213.1 2734.15
   226.5 2732.63   239.8  2732.5   251.9 2733.26   292.6 2732.15   336.7 2732.86
   346.1 2731.86   358.2 2731.78   368.2 2730.87   376.2 2730.28   380.7 2730.95
   394.3 2735.39   402.7 2736.03   407.1 2737.13   415.9 2741.81   420.3 2743.48
   429.1 2745.95   437.9 2750.14   473.2 2765.21   493.8 2775.15   509.1 2782.03
#Mann= 5 ,-1,0
       0      .1       0      80     .06       0     190      .1       0
   368.2    .045       0   380.7      .1       0
#XS Ineff= 2 , 0
           201.8  2740.4
Permanent Ineff=
       F       F
Bank Sta=368.2,380.7
XS Rating Curve= 0 ,0
Exp/Cntr(USF)=0,0
Exp/Cntr=0.3,0.1

Type RM Length L Ch R = 1 ,142149  ,264.5,275.6,285
XS GIS Cut Line= 2
2300527.64339506466202.2946564182300508.32132455 466692.77798485
#Sta/Elev= 30
       0 2736.45    14.9 2733.56    42.9 2730.13      60 2728.91    66.9  2727.8
     107 2727.08     127 2728.21     155 2727.34     183 2729.15   193.82728.022
     199 2727.24   219.22728.083   231.1 2727.96   243.1 2726.64     268 2725.46
   271.1 2725.52   279.1 2727.79   283.1 2728.07   321.9 2727.45   357.8 2728.19
   391.3    2728     412  2729.4   419.2 2731.76   424.5 2734.38   431.2 2738.22
   443.2 2746.33   455.2 2752.33   467.2 2760.23   479.8 2767.63   490.9 2773.05
#Mann= 5 ,-1,0
       0      .1       0      60     .06       0   193.8    .045       0
   219.2     .06       0     250      .1       0
#XS Ineff= 2 , 0
          129.12 2731.14
Permanent Ineff=
       F       F
Bank Sta=193.8,219.2
XS Rating Curve= 0 ,0
Exp/Cntr(USF)=0,0
Exp/Cntr=0.3,0.1

Type RM Length L Ch R = 1 ,141873  ,249.6,232.4,202.3
XS GIS Cut Line= 3
2300369.89400603466149.7753296912300148.42438313466574.757579042
2300142.43871764466691.478055976
#Sta/Elev= 30
       0 2744.09     8.3 2744.48    33.5 2739.38    51.2 2737.76      58 2735.58
      67 2728.82    80.5  2727.8      85 2729.22    89.5 2727.83    98.6 2723.01
   112.1  2724.3   134.6 2723.09   148.2  2724.9   178.7 2722.41   184.3 2721.36
   206.8 2721.25   217.3 2722.44   249.9 2723.36   310.6 2721.23   335.9 2722.56
   378.2 2722.22   404.1 2720.98   421.9 2722.08   468.4 2721.99   481.7  2722.6
   485.6 2723.64   493.7 2726.95   509.7  2736.3   557.5 2766.76   596.1 2787.23
#Mann= 5 ,-1,0
       0      .1       0      10     .06       0     120      .1       0
   178.7    .045       0   217.3      .1       0
#XS Ineff= 2 , 0
          147.55 2728.09
Permanent Ineff=
       F       F
Bank Sta=178.7,217.3
XS Rating Curve= 0 ,0
Exp/Cntr(USF)=0,0
Exp/Cntr=0.3,0.1

Type RM Length L Ch R = 1 ,141641  ,372.5,395.1,408.5
XS GIS Cut Line= 4
2300100.64719395466072.9652087772300045.71422817466203.780969534
 2300142.6882979466429.7005632362300118.90728804466695.750611082
#Sta/Elev= 30
       0 2742.63    13.2 2741.79    43.6 2735.95      48 2733.86    52.3 2730.68
    64.7  2719.4    69.6 2718.02      87 2719.48   107.5 2718.36   147.8 2719.27
   191.3 2718.98     200 2719.63   239.2 2719.32   246.52718.491   256.6 2717.43
   270.42718.324     288 2719.07   304.5 2718.24   313.2 2719.36   333.6 2719.36
     361 2721.12   396.9 2721.23   423.4 2720.15   439.4 2721.38   491.6 2721.42
   535.8 2722.66   548.1 2728.41   604.9 2764.27   626.9 2776.65   654.8 2790.68
#Mann= 7 ,-1,0
       0      .1       0      90     .06       0  201.88      .1       0
   246.5    .045       0   270.4      .1       0  311.88     .12       0
  417.73      .1       0
#XS Ineff= 2 , 0
           86.76 2727.07  361.24         2726.96
Permanent Ineff=
       F       F
Bank Sta=246.5,270.4
XS Rating Curve= 0 ,0
Exp/Cntr(USF)=0,0
Exp/Cntr=0.3,0.1

Type RM Length L Ch R = 1 ,141246  ,358.9,371.5,371.7
XS GIS Cut Line= 4
2299944.92405096466015.0250517172299861.81691728466179.351635894
2299785.45511264466384.4818879052299612.23446597466529.443492686
#Sta/Elev= 30
       0 2729.53      20 2722.59    42.8 2721.18    51.7 2716.86    58.7 2715.25
    74.1 2716.85    87.6 2717.03   127.2 2713.81   136.9 2715.73   186.1 2716.74
   194.6 2715.75   207.4 2712.55     233 2714.56   271.5 2714.41   283.3 2713.65
   297.1 2714.12   301.3 2712.34     305 2711.98   314.1 2711.31   319.72711.936
   331.2  2713.7     361 2713.49   378.2 2717.44   395.2  2716.5     436 2722.41
   509.5 2727.77   541.2 2727.87   580.5 2731.92   603.6 2740.76   628.9 2752.72
#Mann= 8 ,-1,0
       0      .1       0      60     .06       0     160     .12       0
  261.96      .1       0     305    .045       0   319.7      .1       0
  361.96     .12       0  456.78      .1       0
#XS Ineff= 2 , 0
          185.75  2720.8
Permanent Ineff=
       F       F
Bank Sta=305,319.7
XS Rating Curve= 0 ,0
Exp/Cntr(USF)=0,0
Exp/Cntr=0.3,0.1

Type RM Length L Ch R = 1 ,140874  ,268.2,261.8,254.9
XS GIS Cut Line= 4
2299743.79892403 465949.202583792299707.29868439466026.693541475
2299600.03817053466141.9407638672299475.26126692466402.504297863
#Sta/Elev= 30
       0 2723.81     4.4 2721.75    13.2 2715.23    17.7 2712.98    53.8 2712.21
    62.8 2713.27    83.9 2713.44     100 2711.93   121.8 2711.15   129.2 2709.63
   143.1 2708.36   149.1 2704.85   152.62704.623     171 2703.77   180.2 2704.53
   187.4  2705.7   198.3 2709.54   219.8 2711.81   278.4 2711.08   317.4 2709.65
   353.1 2710.01   383.4 2709.14   397.5 2715.62   401.9 2716.99   410.8 2717.79
   459.6 2717.19   472.9 2717.86   483.6 2720.49   490.6 2723.15     532 2742.94
#Mann= 6 ,-1,0
       0      .1       0      10     .06       0  135.66     .12       0
   152.6    .045       0   180.2     .12       0   353.1      .1       0
Bank Sta=152.6,180.2
XS Rating Curve= 0 ,0
Exp/Cntr(USF)=0,0
Exp/Cntr=0.3,0.1

Type RM Length L Ch R = 1 ,140612  ,433.4,434.1,427.8
XS GIS Cut Line= 2
2299456.91172227465907.0665923772299258.73664008466307.086665696
#Sta/Elev= 30
       0 2708.59    24.7 2707.92      29 2706.92      35    2703    37.9 2701.25
    40.9  2700.5    46.9 2700.27    51.5 2700.36    60.4 2702.94    73.8 2703.37
    82.7 2705.22    96.1 2706.64   118.4 2706.37   127.8 2707.84   160.3 2708.06
   176.5 2706.54   199.1 2707.48   212.2 2706.78     226 2704.48   267.8 2706.12
   286.1 2703.88   300.6 2705.99   314.8 2705.68   327.5 2707.47   339.2 2705.05
   350.5 2705.84   372.9 2709.25   386.3 2712.64   408.6 2723.86   446.4 2744.86
#Mann= 4 ,-1,0
       0     .06       0      35    .045       0    60.4     .06       0
     170      .1       0
#XS Ineff= 2 , 0
                          158.59         2713.32
Permanent Ineff=
       F       F
Bank Sta=35,60.4
XS Rating Curve= 0 ,0
Exp/Cntr(USF)=0,0
Exp/Cntr=0.3,0.1

Type RM Length L Ch R = 1 ,140178  ,342.9,342.5,338.4
XS GIS Cut Line= 2
2299133.95973648465787.7945521672298944.95942661466145.610672796
#Sta/Elev= 30
       0 2703.85    12.4 2703.46    28.7 2702.24    42.3 2701.86    55.9 2702.15
      92 2701.55   114.7 2702.38   119.2 2701.77   132.6 2698.18   137.3 2697.55
   141.8  2697.5   159.2 2699.06   182.5  2699.6   205.1  2698.5   217.1  2696.6
   223.2 2696.12   232.3  2696.5   236.8 2697.23   241.3 2698.98   254.9 2698.81
   269.3 2698.03   291.1 2699.66   304.7 2701.61   313.2 2704.13   320.7  2707.1
   336.8  2715.5   348.7 2720.39   381.2 2728.95   395.1 2730.71   404.7 2734.03
#Mann= 4 ,-1,0
       0     .06       0      90      .1       0   217.1    .045       0
   232.3      .1       0
Bank Sta=217.1,232.3
XS Rating Curve= 0 ,0
Exp/Cntr(USF)=0,0
Exp/Cntr=0.3,0.1

Type RM Length L Ch R = 1 ,139836  ,286.7,287.9,291
XS GIS Cut Line= 2
2298872.91540039465679.9247869432298732.10470869466059.367812952
#Sta/Elev= 30
       0 2699.27    18.4 2698.74    31.2 2696.49    56.8 2695.97    86.7 2696.19
   112.3 2695.06   140.1 2696.32   146.4 2695.19   150.7 2693.49   163.4 2691.19
   175.8 2690.94   188.3 2691.32   193.3 2692.92   201.9 2694.23   214.7 2694.86
   240.3 2696.94   253.1 2696.91   261.6  2695.4   266.1 2695.31   274.4 2695.95
   297.2 2695.82   312.7 2693.57   325.6 2695.16   337.6 2695.65   340.7 2696.25
   342.7 2696.84   346.9 2699.05   355.5 2705.16   368.7 2716.76   404.7 2747.29
#Mann= 4 ,-1,0
       0     .06       0      90      .1       0   163.4    .045       0
   188.3      .1       0
#XS Ineff= 2 , 0
                          246.76         2702.74
Permanent Ineff=
       F       F
Bank Sta=163.4,188.3
XS Rating Curve= 0 ,0
Exp/Cntr(USF)=0,0
Exp/Cntr=0.3,0.1

Type RM Length L Ch R = 1 ,139548  ,236.7,237,236.6
XS GIS Cut Line= 2
2298628.06535024465584.1299414722298469.44521492  465943.2698705
#Sta/Elev= 30
       0 2695.71    14.3 2695.19      25 2694.03    36.1 2692.28    46.2 2691.83
    66.7  2692.2    75.5 2693.23    97.3 2691.17   149.8 2690.81   176.1 2691.15
   189.2 2692.24   193.5 2692.05   202.3 2690.85     211 2688.71   219.8 2689.05
   226.22687.375   228.5 2686.93   237.2 2686.85   255.5  2687.3   258.5 2688.13
   267.9 2692.16   272.3 2694.56   279.8 2699.37   285.4 2704.28   294.9  2715.9
   298.5 2719.21   306.6 2724.94   320.4 2733.68   355.3 2754.48   392.6 2775.56
#Mann= 4 ,-1,0
       0     .06       0      90      .1       0   226.2    .045       0
   255.5      .1       0
Bank Sta=226.2,255.5
XS Rating Curve= 0 ,0
Exp/Cntr(USF)=0,0
Exp/Cntr=0.3,0.1

Type RM Length L Ch R = 1 ,139311  ,303.6,299.8,289.2
XS GIS Cut Line= 2
2298403.40286413 465510.255392212298254.77155249465846.052059262
#Sta/Elev= 30
       0 2691.73    11.9 2690.48    20.7 2689.05    33.8  2688.2    95.1 2687.33
   107.8 2687.97   130.1 2685.41   134.4 2685.69   146.3  2687.4   150.2 2687.69
     165 2687.66   183.6 2687.01   195.6 2687.47   204.4 2687.46   208.8 2686.52
   211.82685.288   213.9 2684.66   226.3 2684.37     235 2684.47   238.1 2685.29
   239.4  2685.9   241.2 2687.25     255 2699.88   261.3 2705.03   278.8 2717.91
   292.7 2726.15   304.5 2731.75     320 2738.18   344.4 2746.02   367.2 2752.49
#Mann= 4 ,-1,0
       0     .06       0      60      .1       0   211.8    .045       0
   238.1      .1       0
Bank Sta=211.8,238.1
XS Rating Curve= 0 ,0
Exp/Cntr(USF)=0,0
Exp/Cntr=0.3,0.1

Type RM Length L Ch R = 1 ,139011  ,232.2,206.3,181.8
XS GIS Cut Line= 2
2298217.42434196465459.4259568672298131.30926864465821.304534623
#Sta/Elev= 30
       0 2689.22      10 2688.13    14.1 2687.56    18.2  2685.7      24 2682.16
    26.5 2681.25    29.1 2681.07    43.8 2680.87    51.1  2681.1    56.32682.341
    63.5 2684.85    67.6 2685.24   104.6 2684.79   162.2 2685.83   174.5 2685.09
   195.1 2685.28   203.3 2684.21   211.5 2685.08   223.8 2683.88   232.1 2685.42
   240.3 2685.76   244.4 2687.43   248.3 2690.02   264.9 2703.92   273.2 2709.55
   285.5 2720.58   293.7 2726.36   308.2 2734.45   333.7 2747.25     372 2767.57
#Mann= 4 ,-1,0
       0     .06       0      10      .1       0      24    .045       0
    56.3      .1       0
#XS Ineff= 2 , 0
                          162.17         2688.73
Permanent Ineff=
       F       F
Bank Sta=24,56.3
XS Rating Curve= 0 ,0
Exp/Cntr(USF)=0,0
Exp/Cntr=0.3,0.1

Type RM Length L Ch R = 1 ,138805  ,194.7,212.9,231.6
XS GIS Cut Line= 3
 2297903.7998267465431.4954716342298062.28062321465610.760177832
2298034.36829006465791.404111668
#Sta/Elev= 30
       0 2683.36    48.9 2680.61    63.8 2680.16      77 2681.85   103.2 2681.59
   109.1 2682.33   114.4 2682.45     125 2681.63   133.4 2682.24   146.4 2682.29
   151.5 2680.77   154.5 2678.91   157.3 2677.76   173.1 2677.42   187.8 2678.91
   205.1 2677.53   215.8  2681.5   239.3 2682.29   246.7 2683.37   282.2 2683.18
   294.3 2682.43   310.5 2682.61   314.6 2683.13   318.6  2684.9   327.4 2691.83
   330.8 2694.76     351 2714.38   358.9 2720.51     384 2735.99   422.1 2757.23
#Mann= 5 ,-1,0
       0     .07       0      50      .1       0     120     .06       0
   154.5    .045       0   187.8      .1       0
#XS Ineff= 2 , 0
          133.55 2686.51
Permanent Ineff=
       F       F
Bank Sta=154.5,187.8
XS Rating Curve= 0 ,0
Exp/Cntr(USF)=0,0
Exp/Cntr=0.3,0.1

Type RM Length L Ch R = 1 ,138592  ,140.1,127.7,117.5
XS GIS Cut Line= 2
2297878.85088258465446.4930217212297843.98674775465818.988778068
#Sta/Elev= 30
       0 2682.29    46.9 2681.74    54.9 2681.42      67 2680.02    95.1 2678.77
   111.2 2678.66   123.2 2679.26   135.3 2679.29   147.3 2677.29   155.4 2677.57
   167.4 2676.16     195 2677.15   199.6 2677.04   211.6 2676.08   219.72674.533
     229 2674.11   243.7 2674.19   244.52674.605   251.1 2678.19   259.8 2681.89
   263.8 2684.31   267.9 2687.38   283.9 2702.19   287.9 2705.49     300 2714.34
     312 2722.38   345.7 2743.18   360.3 2751.82   364.9 2754.92   374.1 2760.28
#Mann= 5 ,-1,0
       0     .07       0      20     .06       0     120      .1       0
   219.7    .045       0   244.5      .1       0
#XS Ineff= 2 , 0
           130.1 2682.89
Permanent Ineff=
       F       F
Bank Sta=219.7,244.5
XS Rating Curve= 0 ,0
Exp/Cntr(USF)=0,0
Exp/Cntr=0.3,0.1

Type RM Length L Ch R = 1 ,138464  ,296.6,300.7,303
XS GIS Cut Line= 2
2297627.46212091 465453.832839582297792.60802273465817.153823604
#Sta/Elev= 30
       0 2681.26    21.2 2681.16    30.3 2681.58    60.5  2681.1   166.4 2676.78
   223.4 2676.91   229.6 2676.49   235.7 2675.32   240.9 2673.67   244.7  2671.9
     253 2671.41   265.9 2671.53   268.9 2671.97   271.7 2672.79   276.1 2674.73
   280.5 2675.44   284.9 2675.42   289.3  2674.7   293.1 2674.64   298.1 2675.33
   302.5 2677.86   306.9 2683.02   311.2 2688.89   317.2 2695.69   324.4 2702.73
   328.8  2706.7     342 2717.24   350.8 2723.45   390.3 2747.57   399.1 2752.49
#Mann= 5 ,-1,0
       0     .06       0      20     .05       0     150      .1       0
   244.7    .045       0   268.9      .1       0
#XS Ineff= 2 , 0
          222.45 2680.07
Permanent Ineff=
       F       F
Bank Sta=244.7,268.9
XS Rating Curve= 0 ,0
Exp/Cntr(USF)=0,0
Exp/Cntr=0.3,0.1

Type RM Length L Ch R = 1 ,138163  ,227.6,241.6,253.2
XS GIS Cut Line= 2
2297368.73354137465499.7067011992297480.66576372  465885.0471388
#Sta/Elev= 30
       0 2676.43     9.9 2676.09    26.5 2676.44      39 2675.96    59.8 2676.97
    97.3    2675     139  2675.6   147.3 2675.03   180.6 2673.99   197.3 2674.43
   226.7  2672.8   247.3 2672.63   252.5 2672.25   262.2 2672.57   268.1 2671.89
   279.82669.014     288 2667.83   296.5 2667.59   305.6 2667.96   308.3 2668.78
   309.8 2669.23   313.5 2675.29   318.1 2686.67   322.3 2695.28   326.7 2700.24
   334.8 2707.73   342.1 2713.55   351.4 2719.98     367 2729.44   401.3 2751.38
#Mann= 5 ,-1,0
       0     .05       0      80     .06       0     170      .1       0
   279.8    .045       0   308.3      .1       0
#XS Ineff= 2 , 0
             260 2679.22
Permanent Ineff=
       F       F
Bank Sta=279.8,308.3
XS Rating Curve= 0 ,0
Exp/Cntr(USF)=0,0
Exp/Cntr=0.3,0.1

Type RM Length L Ch R = 1 ,137922  ,424.6,435.6,444.8
XS GIS Cut Line= 2
2297280.65572706465477.687247622 2297185.2380949465877.707320941
#Sta/Elev= 30
       0 2675.48    13.3 2675.72    36.5 2674.35    52.9 2674.06    77.6 2675.89
   143.4  2672.7     164 2672.29   179.3 2674.19   192.8 2673.19   208.9 2674.95
   213.3 2674.92   225.6 2669.08   229.8 2668.41     238 2668.38   258.5 2669.29
   266.8 2665.62   271.52664.997   295.5  2664.5   304.82665.262   307.9  2666.7
   308.8 2667.73   315.4 2676.63   324.3 2689.93   329.6 2696.24   340.8 2707.93
     349 2714.47   357.2 2718.79   361.4 2720.26   382.1 2724.97   411.2 2733.58
#Mann= 4 ,-1,0
       0     .05       0     200      .1       0   271.5    .045       0
   304.8      .1       0
#XS Ineff= 2 , 0
          253.52 2674.97
Permanent Ineff=
       F       F
Bank Sta=271.5,304.8
XS Rating Curve= 0 ,0
Exp/Cntr(USF)=0,0
Exp/Cntr=0.3,0.1

Type RM Length L Ch R = 1 ,137486  ,669,659.8,652.3
XS GIS Cut Line= 2
2296928.00497401465413.8473593512296724.12114459465728.734607008
#Sta/Elev= 30
       0 2665.31      37 2664.09    65.9 2664.47    99.3 2665.52   141.1 2665.13
   172.9 2666.05   175.8 2665.75   180.3 2660.78   183.7 2658.31     185 2657.54
   190.3  2656.3   213.1 2656.16   223.2 2656.34   229.92658.255   236.6 2660.63
   242.4 2661.17     247 2662.13   251.8 2665.18   256.5 2667.25   275.6 2667.44
   282.2 2668.23   288.6 2668.44   294.7 2667.35   299.4 2667.06   301.4  2667.9
     306 2670.25   311.8 2674.11   346.5 2701.83   360.3 2711.66   375.1 2721.62
#Mann= 4 ,-1,0
       0     .05       0     180      .1       0   183.7    .045       0
   229.9      .1       0
Bank Sta=183.7,229.9
XS Rating Curve= 0 ,0
Exp/Cntr(USF)=0,0
Exp/Cntr=0.3,0.1

Type RM Length L Ch R = 1 ,136826  ,500.5,496.1,492.7
XS GIS Cut Line= 2
2296271.04596811465117.0831187542296173.63480516465488.604763471
#Sta/Elev= 30
       0 2654.34    37.3 2653.82    58.1 2655.75    90.9 2653.97   103.5 2656.69
   115.9 2658.59   128.3  2659.1   153.1 2658.72   157.2 2658.08   161.4  2655.6
   169.6 2649.38   177.52646.946     182 2646.16   189.2 2646.04   198.6 2646.09
   202.7 2646.92   206.9    2649     211 2652.86   215.4 2655.75   227.5 2655.21
   235.8 2655.97   244.9  2654.8   260.6  2654.4   281.3 2654.93   289.6 2656.89
   306.1 2657.35   330.9 2656.38   333.3 2656.88   339.9 2659.66   384.1 2688.07
#Mann= 5 ,-1,0
       0      .1       0      60     .06       0   177.5    .045       0
   202.7     .06       0     250      .1       0
Bank Sta=177.5,202.7
XS Rating Curve= 0 ,0
Exp/Cntr(USF)=0,0
Exp/Cntr=0.3,0.1

Type RM Length L Ch R = 1 ,136330  ,533,534,533.3
XS GIS Cut Line= 2
2295752.27489103464965.3029346312295716.02887692465420.643486999
#Sta/Elev= 30
       0 2653.03      44 2652.91   100.2 2650.63   104.2 2650.02   116.2 2645.57
   124.3  2645.1   140.3 2647.54   200.5  2647.1   204.7 2647.42   212.5  2650.1
   215.6  2650.4   240.6 2650.73   252.6  2649.2   260.7 2645.83   282.5 2642.04
   292.62639.547   308.8 2638.41   320.9 2638.44   324.9 2639.52   332.9 2645.56
   336.9 2647.24     345 2648.74   377.1  2648.2   397.1 2646.23   405.2 2646.67
   409.2 2649.03   416.3    2655   433.2 2672.67   437.3 2676.31   456.8 2691.01
#Mann= 5 ,-1,0
       0     .12       0      10      .1       0     110     .06       0
   292.6    .045       0   324.9      .1       0
Bank Sta=292.6,324.9
XS Rating Curve= 0 ,0
Exp/Cntr(USF)=0,0
Exp/Cntr=0.3,0.1

Type RM Length L Ch R = 1 ,135796  ,406.5,408.5,409.9
XS GIS Cut Line= 2
2295238.03456572464849.7687646272295188.19629631465391.193600527
#Sta/Elev= 30
       0 2644.72    31.5  2644.1    67.4 2641.98     148 2639.79   180.2 2640.82
   196.2 2639.21   208.3 2638.86   268.5 2640.65   280.6 2641.91   300.7 2641.92
   320.8 2640.02   324.9 2638.57   334.32633.217   336.8 2632.46   352.9 2632.02
   371.3 2633.25     381 2637.14     389 2637.36   401.1 2639.47   433.2  2640.6
   453.6 2639.22   469.4 2640.14   481.4 2642.28   501.5 2641.56   513.6 2640.19
   517.6 2640.53   521.6 2642.07   527.2 2645.85   533.7 2651.27   543.7 2660.83
#Mann= 5 ,-1,0
       0     .05       0     230     .06       0     330      .1       0
   334.3    .045       0   371.3      .1       0
Bank Sta=334.3,371.3
XS Rating Curve= 0 ,0
Exp/Cntr(USF)=0,0
Exp/Cntr=0.3,0.1

Type RM Length L Ch R = 1 ,135388  ,406.7,403.6,399
XS GIS Cut Line= 3
2294884.03159011464605.4736348682294767.31111318465374.631649538
2294830.16060076465554.201614052
#Sta/Elev= 30
       0 2652.05    40.2 2647.68   164.7 2640.01   246.5 2636.92   262.7  2634.3
   274.8 2631.33     295 2630.05   347.6 2634.04   364.9  2633.5     469 2634.31
   498.4 2635.76   517.6 2635.15   521.6 2633.76   527.52629.158   533.7 2626.35
   548.3 2625.82     558 2626.25   562.1  2628.9   566.1 2631.08   582.3 2634.07
   598.5 2633.22   671.3  2632.8   707.7 2635.46   758.2 2635.26   776.5 2637.47
   801.9 2647.69   852.8 2671.77   878.1 2681.49   903.6 2695.06   968.2 2731.89
#Mann= 6 ,-1,0
       0     .05       0     480     .06       0   527.5    .045       0
   562.1     .06       0     580     .05       0  777.96      .1       0
#XS Ineff= 2 , 0
          492.39 2648.19
Permanent Ineff=
       F       F
Bank Sta=527.5,562.1
XS Rating Curve= 0 ,0
Exp/Cntr(USF)=0,0
Exp/Cntr=0.3,0.1

Type RM Length L Ch R = 1 ,134984  ,373.4,374.6,374.6
XS GIS Cut Line= 4
2294501.59150311464601.6093538962294404.49609088  464806.3903218
 2294399.8444471465337.8720228312294398.17169392465584.737373791
#Sta/Elev= 30
       0 2646.98    72.8 2639.37   127.9 2634.97   167.7  2632.7   241.4 2630.73
   253.5 2629.21   269.4  2625.5   289.4 2624.06   305.4 2624.15   325.4  2627.4
   337.4 2628.13   401.4 2628.82   447.8 2626.52   481.4  2628.8   501.4 2628.14
   529.4 2622.73   545.4 2621.43     552 2622.75   557.4 2625.87   561.4 2626.98
   753.4 2629.18     790 2628.32   813.4 2629.32   837.4  2639.6   845.4 2640.97
   849.4  2642.7   865.4 2653.72   890.7 2667.96   955.8 2707.11    1005 2739.17
#Mann= 8 ,-1,0
       0      .1       0      80     .05       0     280     .03       0
     380     .06       0     480     .05       0   529.4    .045       0
     552     .05       0     790      .1       0
#XS Ineff= 2 ,-1
       0  468.17 2640.05  607.32     996  2639.3
Permanent Ineff=
       F       F
Bank Sta=529.4,552
XS Rating Curve= 0 ,0
Exp/Cntr(USF)=0,0
Exp/Cntr=0.3,0.1

Type RM Length L Ch R = 1 ,134610  ,327.7,307.9,292.5
XS GIS Cut Line= 2
2294059.70708564464564.6830155342294007.93546157465601.873557592
#Sta/Elev= 30
       0 2642.13    24.5 2640.94    84.6 2642.26   140.7  2637.6   184.7  2636.6
   208.8  2632.6   232.7 2625.91   280.8 2621.28   312.9    2620   360.9 2622.13
     429 2621.56   461.1 2623.85   485.1 2622.85   489.1 2621.85   493.1 2619.56
   505.1 2618.66   527.9 2619.48   541.2 2621.94   557.2 2622.65   613.3 2619.24
   649.3 2621.01   725.4 2621.22   817.5 2624.49   909.6  2625.6   933.7 2633.87
   953.7 2644.04   965.7 2651.51   977.7 2654.25   993.7 2664.44  1038.5 2689.21
#Mann= 8 ,-1,0
       0      .1       0      20     .05       0     120     .06       0
     220     .05       0     410     .07       0   493.1    .045       0
   527.9     .05       0     910      .1       0
#XS Ineff= 2 , 0
          454.31 2632.21
Permanent Ineff=
       F       F
Bank Sta=493.1,527.9
XS Rating Curve= 0 ,0
Exp/Cntr(USF)=0,0
Exp/Cntr=0.3,0.1

Type RM Length L Ch R = 1 ,134302  ,267,264.3,259.7
XS GIS Cut Line= 4
2293651.95744156464616.3813833862293676.45582382465082.064407904
2293875.44695609465350.688987603 2293926.3251127465626.029599858
#Sta/Elev= 30
       0 2638.88    28.8 2631.81    44.9 2631.08   100.9  2623.2     145  2620.3
   297.2 2618.81   325.2 2617.26   345.3 2618.82   381.3 2619.75   401.4 2616.59
   413.4  2619.7     515 2619.31   529.9 2616.45   591.3 2617.91   608.5 2617.35
  612.23 2616.81   619.9 2615.77   627.1 2616.84   639.5 2619.35   659.4 2616.07
   729.1 2617.96     775  2621.3   929.3 2622.84   941.5 2623.16   961.8 2630.11
   982.5 2639.23  1010.6 2655.65  1022.8 2658.53    1035 2667.73  1080.6 2694.86
#Mann= 8 ,-1,0
       0      .1       0     145     .05       0   345.3     .06       0
   591.3      .1       0   608.5     .05       0  612.23    .045       0
   627.1     .05       0   929.3      .1       0
#XS Ineff= 2 , 0
           470.2 2626.88
Permanent Ineff=
       F       F
Bank Sta=612.23,627.1
XS Rating Curve= 0 ,0
Exp/Cntr(USF)=0,0
Exp/Cntr=0.3,0.1

Type RM Length L Ch R = 1 ,134038  ,562.6,577.5,592.5
XS GIS Cut Line= 4
 2293384.9109569464660.4332108852293419.82370644465231.755370497
2293718.16408095465501.0683782632293760.11548618465668.873999183
#Sta/Elev= 30
       0 2661.87    32.8 2641.86    56.7 2630.04    60.9 2628.83    84.9 2624.53
   172.3  2615.6   249.3 2615.06   301.3 2616.89   337.4 2614.35   411.3 2611.89
   551.4 2612.98   574.5 2613.97   586.5    2612   594.4 2611.77   642.9  2613.8
   672.8 2613.42   705.8 2614.56   718.1  2613.4   757.7 2612.44   771.5 2610.74
776.0416 2612.24   799.2 2615.51   819.3  2615.2   982.6 2619.05     995 2623.31
  1026.7 2639.11  1065.1 2663.21  1077.5 2666.36  1089.9 2676.73  1147.3 2713.47
#Mann= 8 ,-1,0
       0      .1       0  272.87     .06       0  292.87     .08       0
  692.87      .1       0   757.7    .045       0776.0416      .1       0
  962.87     .05       0 1115.37      .1       0
Bank Sta=757.7,776.0416
XS Rating Curve= 0 ,0
Exp/Cntr(USF)=0,0
Exp/Cntr=0.3,0.1

Type RM Length L Ch R = 1 ,133460  ,578.9,581.2,583
XS GIS Cut Line= 3
2293022.58940812464810.7388470922293001.73758593 465124.83498558
2293066.51891971465733.199487202
#Sta/Elev= 30
       0 2620.34    50.6 2616.18    86.6 2614.15    94.6 2612.63   102.7  2613.4
   126.7 2612.66   146.8 2610.12     271 2610.58   334.9 2607.89   367.4 2607.47
   415.5 2605.45     468  2605.3   519.5 2606.59   584.6  2605.8     653 2606.88
   729.5 2605.84747.57512603.115   769.7 2602.65  774.63 2603.18   777.7  2604.2
   781.8 2607.15   797.8 2624.75   813.9 2638.46   822.6 2644.62   862.2 2670.42
   873.5 2679.54   878.3 2681.49   886.3 2683.06   902.4 2694.78   926.6 2707.21
#Mann= 4 ,-1,0
       0     .06       0      40     .08       0747.5751    .045       0
  774.63      .1       0
Bank Sta=747.5751,774.63
XS Rating Curve= 0 ,0
Exp/Cntr(USF)=0,0
Exp/Cntr=0.3,0.1

Type RM Length L Ch R = 1 ,132879  ,412.6,436.5,460.3
XS GIS Cut Line= 2
2292465.21544474465095.5381277052292481.99600683465811.508776965
#Sta/Elev= 30
       0 2604.03    77.7 2602.94   173.7 2602.62   221.7 2600.93   241.7  2599.8
   293.6 2599.13   341.7 2597.01   409.8 2598.45   446.3 2600.13   485.8 2599.47
   501.8 2599.63   513.8 2600.17   517.8 2599.66   526.72596.718   529.8 2596.28
   541.8 2596.02   553.8 2596.19   556.72596.569   557.8 2596.71   577.8 2614.75
   588.6 2624.96   598.7 2633.38   609.8 2642.19   614.4 2645.13   625.8 2653.32
   633.7  2657.9   661.8 2675.84   680.8 2686.25   701.8 2696.17   716.2 2701.38
#Mann= 4 ,-1,0
       0     .05       0     470      .1       0   526.7    .045       0
   556.7      .1       0
#XS Ineff= 2 , 0
          451.84  2603.2
Permanent Ineff=
       F       F
Bank Sta=526.7,556.7
XS Rating Curve= 0 ,0
Exp/Cntr(USF)=0,0
Exp/Cntr=0.3,0.1

Type RM Length L Ch R = 1 ,132442  ,371.5,350.4,316
XS GIS Cut Line= 4
 2292140.7912443465098.3348880542292151.97828569465405.978526408
2292042.90463209465498.2716179142292054.09167349465817.102297663
#Sta/Elev= 30
       0 2599.89    82.9 2597.62   134.9  2597.4     191  2593.7     259 2594.58
     283 2594.22   312.8 2595.28   324.2  2593.9   352.6 2593.85   371.42591.833
   399.5 2591.32   409.3 2591.69   418.1  2593.3   485.7 2592.66   513.7 2593.21
   545.7 2592.42   557.7 2593.32   569.7 2591.93   585.7 2591.96   589.7 2592.62
   597.6  2597.3   610.1 2606.92   617.2 2613.06   629.7 2625.38   643.2 2637.29
   661.8 2652.44     693  2674.7   715.1  2689.7   733.8 2703.41   769.8 2726.45
#Mann= 5 ,-1,0
       0     .03       0      80     .05       0   371.4    .045       0
   409.3     .05       0  520.73      .1       0
#XS Ineff= 2 , 0
          304.27 2599.16
Permanent Ineff=
       F       F
Bank Sta=371.4,409.3
XS Rating Curve= 0 ,0
Exp/Cntr(USF)=0,0
Exp/Cntr=0.3,0.1

Type RM Length L Ch R = 1 ,132092  ,270.5,278.4,280.5
XS GIS Cut Line= 2
2291796.78972141465006.041796547 2291807.9767628465791.931454525
#Sta/Elev= 30
       0 2600.97    67.1 2599.18   147.2 2594.77   223.4  2591.8   255.2 2589.67
   258.9 2588.43   271.2 2587.12   283.2 2587.12   304.1 2588.56   315.2 2589.72
   343.2 2588.82   367.2 2589.93   411.2 2589.33   427.2 2590.72   455.2 2590.86
   479.2 2589.25   495.2 2590.19   539.2 2588.31   543.2 2588.51   555.2 2591.42
   559.2 2591.55   575.2  2591.3   591.2 2589.75   611.2 2589.15   631.2 2593.27
   639.2 2596.06   647.2 2600.79   683.2 2628.65   766.7 2688.54     786  2701.7
#Mann= 7 ,-1,0
       0     .03       0     170     .05       0   258.9    .045       0
   304.1     .05       0     370     .07       0     460     .05       0
     660      .1       0
#XS Ineff= 2 , 0
                          514.29         2600.83
Permanent Ineff=
       F       F
Bank Sta=258.9,304.1
XS Rating Curve= 0 ,0
Exp/Cntr(USF)=0,0
Exp/Cntr=0.3,0.1

Type RM Length L Ch R = 1 ,131814  ,390.3,390.5,393.5
XS GIS Cut Line= 3
2291649.02691461464954.0733064872291524.92696283465387.938390043
2291513.93086513465796.218044716
#Sta/Elev= 30
       0 2601.05    98.9 2600.07   198.8 2597.72   207.1 2596.65   227.9 2589.36
   244.5 2587.44   279.5 2585.88   362.3 2587.24   384.2 2585.98   394.3 2585.47
     413 2585.99   419.3 2586.85   472.5 2586.41   484.5 2585.75   520.5  2587.5
   532.5 2587.27   544.5  2585.8   552.5  2586.2   560.5 2584.98   568.5  2586.3
   584.6 2586.55   600.6    2588   651.9 2586.52   680.6 2588.45   708.6 2588.05
   716.6 2589.65   728.6 2594.14   737.7 2598.65   780.5 2623.82   859.7 2676.89
#Mann= 6 ,-1,0
       0     .05       0     330     .07       0   384.2    .045       0
     413     .07       0     440     .05       0     740      .1       0
#XS Ineff= 2 , 0
                          602.78         2590.56
Permanent Ineff=
       F       F
Bank Sta=384.2,413
XS Rating Curve= 0 ,0
Exp/Cntr(USF)=0,0
Exp/Cntr=0.3,0.1

Type RM Length L Ch R = 1 ,131423  ,402,386.6,370.7
XS GIS Cut Line= 3
 2291375.7275059464764.6745863882291175.29972528465381.313671111
2291164.93837093465816.379821496
#Sta/Elev= 30
       0  2604.7    13.1 2604.65      30 2608.35   196.8 2598.31   286.5 2595.21
   307.6 2592.98   311.8 2591.15     316 2587.39   320.2 2580.75     337 2580.03
   347.2 2580.75     358  2582.8   371.4 2582.26     400 2584.08   421.1 2582.74
   488.4 2582.52   538.9  2580.9   559.9 2583.35   576.8 2583.22   593.6 2582.47
     602 2580.91   615.9 2580.76   660.3 2584.94   824.3 2584.48   904.3 2585.77
   932.7 2587.29   956.3 2590.71   976.4 2597.24   992.4 2604.68  1083.6 2657.25
#Mann= 10 ,-1,0
       0     .07       0      20     .06       0     120     .05       0
     290     .08       0   320.2    .045       0   347.2      .1       0
     540     .05       0     610      .1       0     640     .05       0
 1038.39      .1       0
Bank Sta=320.2,347.2
XS Rating Curve= 0 ,0
Exp/Cntr(USF)=0,0
Exp/Cntr=0.3,0.1

Type RM Length L Ch R = 1 ,131037  ,176,212.5,217.1
XS GIS Cut Line= 4
2290888.59987967464697.652883319 2290869.7450334465058.588511993
 2290990.3165923465253.886172582 2291024.9885069465819.787149342
#Sta/Elev= 30
       0 2600.14    23.6 2599.89    51.6 2596.92    79.6 2595.16   119.7 2594.35
   175.8 2594.53   187.8 2594.15   215.8 2591.62     356 2588.79     360 2588.17
   383.3 2578.43   391.2 2577.72   408.7 2577.89   420.3 2576.77     435 2577.05
     4512574.683   458.5 2573.87   472.82574.633   487.9 2578.57   503.1 2579.61
   622.4  2580.5   762.6 2582.67   950.9 2583.06  1007.4 2583.85  1031.1 2585.12
    1045 2587.71  1067.1 2595.71  1082.9 2604.36  1124.5 2625.36  1157.9 2644.41
#Mann= 9 ,-1,0
       0     .08       0      80     .07       0     180     .05       0
     280     .08       0  381.43      .1       0     451    .045       0
   472.8      .1       0  501.43     .05       0 1124.65      .1       0
Bank Sta=451,472.8
XS Rating Curve= 0 ,0
Exp/Cntr(USF)=0,0
Exp/Cntr=0.3,0.1

Type RM Length L Ch R = 1 ,130824  ,335.5,321.9,309.9
BEGIN DESCRIPTION:
start of detailed reach
END DESCRIPTION:
XS GIS Cut Line= 2
 2290747.2930013464721.8340421372290698.80911088465853.124818577
#Sta/Elev= 30
       0 2599.71    27.4 2599.64    71.5 2597.34    95.4 2595.61   139.5 2591.04
   175.1 2589.41   271.6 2586.84   303.6 2586.01   311.6 2586.56   339.7 2577.73
   351.7 2575.97   407.7 2577.18   439.7 2572.54   451.5 2571.67   455.8 2571.36
   467.8 2571.07   471.8 2571.33   475.8 2571.52   486.1 2574.93   507.8 2577.07
     544 2576.75   655.9 2578.96     768 2578.05   988.3 2579.58  1012.1 2580.27
  1025.1 2581.45  1040.3 2584.47  1052.3  2587.9  1092.7 2605.04  1132.3 2625.73
#Mann= 6 ,-1,0
       0     .06       0    71.5     .05       0   271.6     .08       0
   451.5     .05       0   455.8    .045       0   471.8     .05       0
#Block Obstruct= 1 ,-1
   30.93   94.46 2619.52
Bank Sta=455.8,471.8
XS Rating Curve= 0 ,0
Exp/Cntr(USF)=0,0
Exp/Cntr=0.3,0.1

Type RM Length L Ch R = 1 ,130502  ,230.1,254.5,267.5
XS GIS Cut Line= 4
2290437.26462587464718.5846793572290349.88998613465066.669160396
2290519.69228431465561.4617862432290384.61203397465805.915256268
#Sta/Elev= 30
       0 2593.65    68.7 2589.42   134.6 2586.72   163.5 2582.68   184.1 2581.59
   365.7 2577.28   420.7 2580.09   471.5 2580.95   479.9 2579.79   492.6 2573.12
   505.3 2569.93   509.6  2569.4   522.2 2570.74     5392569.462   551.8 2568.62
     573 2568.65   574.42569.512   577.2 2571.37   581.4 2572.09   615.3 2570.96
     637 2573.78   863.3 2577.16   969.7 2576.84  1005.1 2579.59  1018.8 2582.97
  1027.9 2583.78  1041.6 2588.33  1055.3 2596.85  1119.3    2630  1161.3 2648.68
#Mann= 4 ,-1,0
       0     .04       0      50     .05       0     539    .045       0
   574.4     .05       0
#Block Obstruct= 4 ,-1
       0    7.06 2613.65   46.23   60.67 2611.95  182.16  224.04 2601.66
  265.62  304.17 2599.74
Bank Sta=539,574.4
XS Rating Curve= 0 ,0
Exp/Cntr(USF)=0,0
Exp/Cntr=0.3,0.1

Type RM Length L Ch R = 1 ,130248  ,272.2,274.3,273.7
BEGIN DESCRIPTION:
xs 4
END DESCRIPTION:
XS GIS Cut Line= 2
2290231.05059579464694.9306259752290110.20292641465706.598258273
#Sta/Elev= 30
       0  2588.1    34.5 2589.11    87.4 2588.77   123.1 2586.51   191.4 2580.92
   272.2 2576.02   296.1 2575.25   300.4 2574.52   308.4 2572.03   312.5 2571.74
   372.9 2571.16   397.3 2569.67   433.3 2569.98   461.5 2567.59   526.4 2569.57
   540.8 2568.77   614.6 2568.75   630.7 2570.12   707.2 2570.99   743.5 2570.44
   803.9 2570.52   844.2 2572.05   920.7 2572.83   940.9 2573.55   977.1 2576.54
   981.2 2577.69   997.3 2584.94  1009.4 2591.77  1013.4 2593.34  1018.9  2593.8
#Mann= 3 ,-1,0
       0     .05       0   540.8    .045       0   614.6     .05       0
#XS Ineff= 2 , 0
          423.89 2572.39  704.45         2572.76
Permanent Ineff=
       F       F
#Block Obstruct= 1 ,-1
   66.66   99.13 2609.07
Bank Sta=540.8,614.6
XS Rating Curve= 0 ,0
Exp/Cntr(USF)=0,0
Exp/Cntr=0.5,0.3

Type RM Length L Ch R = 1 ,129973  ,172.4,169.8,168.5
BEGIN DESCRIPTION:
Structure XS3 - channel burned within banks
LOB IFA added to uncross profiles at this XS
END DESCRIPTION:
XS GIS Cut Line= 3
2289881.19646125464624.731045109 2289959.5243019464796.284230702
2289826.84439025 465670.49988083
#Sta/Elev= 30
       0 2584.63    13.7 2578.87    31.3 2580.05    48.9 2579.55    59.9 2578.96
    70.8 2580.75    99.2 2581.83   135.4 2578.95   158.8 2577.06   201.6 2570.04
   343.2 2566.26   375.6 2566.01   409.8 2567.29   438.2 2568.16   481.4 2565.96
   549.6 2567.83   606.2 2566.47  606.33 2566.12  606.47 2562.78   606.6 2559.79
  651.14 2564.46  672.41 2562.82  673.11 2563.59   683.1 2567.36   699.3 2568.93
   873.8 2567.35   908.9 2569.38   950.1  2569.9  1010.6 2570.25  1072.8 2573.15
#Mann= 10 ,-1,0
       0     .03       0    13.7    .016       0    48.9     .03       0
   135.4     .05       0   409.8     .04       0   549.6     .03       0
  606.47    .045       0  673.11     .04       0   950.1     .05       0
  1010.6     .04       0
#XS Ineff= 3 ,-1
  166.99  436.06 2570.79  436.06     545  2568.7     723  1072.8    2571
Permanent Ineff=
       F       F       F
#Block Obstruct= 3 ,-1
   89.54  149.28 2600.96  335.91  384.38 2586.54   921.4  939.06 2589.36
Bank Sta=606.47,673.11
XS Rating Curve= 0 ,0
Exp/Cntr(USF)=0,0
Exp/Cntr=0.5,0.3
