HEC-RAS study KNAPPCK.prj: KNAPPCK

--- KNAPPCK.g01 (geometry) --- (continued)

Type RM Length L Ch R = 1 ,32311   ,603.8,594,482.7
XS GIS Cut Line= 2
2244799.49223529437922.4293389572245584.14582105438866.134327233
#Sta/Elev= 30
       0 2303.89    42.2 2277.27    59.2 2263.15    71.2 2262.41    94.9 2244.32
   164.8 2206.84   176.3 2202.26   270.1 2200.16   395.2 2200.66   432.8 2198.48
   454.1 2199.62   462.6 2198.94   470.12195.717   556.3 2195.54   607.4 2200.09
   627.3 2198.42   695.5 2200.81   755.1 2198.07   815.1 2198.71   856.7 2193.97
   942.6 2196.06   962.5 2203.34   990.9 2202.83   996.6 2205.29  1007.6 2215.21
  1013.6 2225.53    1018  2230.4  1168.8 2332.44  1202.3 2353.59  1227.3 2366.86
#Mann= 8 ,-1,0
       0      .1       0   470.1     .04       0   556.3      .1       0
   607.4     .06       0   815.1      .1       0     960    .016       0
   990.9     .06       0    1018      .1       0
#XS Ineff= 2 , 0
          320.08 2210.48   966.2         2212.66
Permanent Ineff=
       F       F
Bank Sta=470.1,556.3
XS Rating Curve= 0 ,0
Exp/Cntr(USF)=0,0
Exp/Cntr=0.3,0.1

Type RM Length L Ch R = 1 ,31717   ,243.6,237.9,199.8
XS GIS Cut Line= 2
2244580.35474738438654.0657905422245304.92224774439131.219998097
#Sta/Elev= 30
       0 2257.75    47.7 2249.35    76.4 2247.18   114.7 2239.47   138.7 2222.51
   163.8 2199.36   179.42193.866     262 2193.52   272.8 2196.24   306.3 2197.28
   348.6  2196.2   363.8 2192.45   387.7 2197.31   440.4 2195.62     450  2192.9
   473.9  2192.8   488.3 2195.66   521.8 2197.18   550.6  2197.5   560.1 2194.89
     571 2194.42   579.3 2196.42   588.9 2202.12   598.5 2203.23   622.4 2201.46
     632 2207.88   646.1 2223.03   686.5 2248.96     802  2304.7   867.6 2333.16
#Mann= 5 ,-1,0
       0      .1       0   179.4     .04       0     262      .1       0
   598.5    .016       0   622.4      .1       0
#XS Ineff= 2 , 0
                          597.18         2211.96
Permanent Ineff=
       F       F
Bank Sta=179.4,262
XS Rating Curve= 0 ,0
Exp/Cntr(USF)=0,0
Exp/Cntr=0.3,0.1

Type RM Length L Ch R = 1 ,31479   ,367.1,353.1,275.7
XS GIS Cut Line= 3
   2244436.53148438877.1837980542245057.82726279439185.098716799
 2245243.6694031439225.182315689
#Sta/Elev= 30
       0 2253.06    89.3  2240.4   111.2 2240.33   129.1 2233.49   162.1 2208.28
   178.2 2198.58   199.7 2196.09     205  2192.2   271.9  2191.6   283.3 2192.16
   325.5 2196.59   365.7 2195.04   381.8 2192.33   402.7 2195.49   450.4 2196.53
   468.4 2192.63   516.1 2193.02   528.1 2196.05   551.9 2194.77   575.5 2197.29
   611.6 2193.86   620.1 2194.64   633.5 2201.46   657.6 2201.17   664.8 2201.56
   682.6 2218.83   692.2 2224.94   773.6 2262.41   859.5 2309.02   883.5 2319.83
#Mann= 5 ,-1,0
       0      .1       0     205     .04       0   283.3      .1       0
   633.5    .016       0   657.6      .1       0
#XS Ineff= 2 , 0
                          633.24         2212.01
Permanent Ineff=
       F       F
Bank Sta=205,283.3
XS Rating Curve= 0 ,0
Exp/Cntr(USF)=0,0
Exp/Cntr=0.3,0.1

Type RM Length L Ch R = 1 ,31126   ,231.2,250.4,300.1
XS GIS Cut Line= 2
2244308.12575386439285.0956572452245223.81780749439416.660607478
#Sta/Elev= 30
       0 2263.46    84.9 2248.47   214.2 2229.52   219.2 2227.69   234.4 2214.62
   254.8 2202.02   262.7 2195.37   274.42190.222   320.9 2189.49   339.5 2189.97
   347.6 2191.91   375.9 2191.08     392 2194.42   416.3 2194.79   472.9 2194.44
   493.1 2192.81   509.2 2193.82   537.5 2191.66     586 2202.67   602.2 2199.41
   613.4 2199.83   655.9 2199.55   666.8  2198.8   670.9  2200.1   691.1 2216.53
   712.5 2229.24   759.8 2251.13   864.8 2304.92     885 2313.26   925.1 2324.58
#Mann= 7 ,-1,0
       0      .1       0   274.4     .04       0   339.5      .1       0
     470     .08       0   613.4    .016       0   655.9      .1       0
   925.1      .1       0
#XS Ineff= 2 , 0
                          590.99         2214.17
Permanent Ineff=
       F       F
Bank Sta=274.4,339.5
XS Rating Curve= 0 ,0
Exp/Cntr(USF)=0,0
Exp/Cntr=0.3,0.1

Type RM Length L Ch R = 1 ,30875   ,282.3,279.1,274.5
BEGIN DESCRIPTION:
Sudden contraction in the floodplain, updated the coefficents to 0.3 and 0.5
END DESCRIPTION:
XS GIS Cut Line= 3
2244270.73113914439403.736528926 2244837.3674689439735.337210651
2244897.49286723439893.849624443
#Sta/Elev= 30
       0 2267.08    50.4 2255.59   151.2 2237.58   171.7 2234.96   186.3  2230.6
   205.6 2230.17   210.2  2228.8   227.2 2220.72   233.1 2219.81   240.4 2216.83
   265.8 2198.48   272.1 2194.75   284.4 2189.33   302.9 2188.16   332.5 2188.07
   367.8 2189.15   395.6  2192.4   420.2 2193.12   437.7  2199.6   455.9 2204.43
   469.8 2202.32   506.8 2200.95   548.6  2202.2   557.8 2201.67   613.2 2205.24
   642.4 2203.95   709.8 2218.98   748.3 2226.45   788.5 2231.73   826.1 2233.47
#Mann= 5 ,-1,0
       0      .1       0   284.4     .04       0   367.8      .1       0
   613.2    .016       0   642.4      .1       0
#XS Ineff= 2 , 0
                           456.9         2212.41
Permanent Ineff=
       F       F
Bank Sta=284.4,367.8
XS Rating Curve= 0 ,0
Exp/Cntr(USF)=0,0
Exp/Cntr=0.5,0.3

Type RM Length L Ch R = 1 ,30596   ,570,561.9,535.3
XS GIS Cut Line= 2
2244151.74124354 439678.375308812244993.75692503440104.645747565
#Sta/Elev= 30
       0 2259.97    22.9 2252.73    41.6 2249.01   100.6 2242.72     175 2231.34
   192.9  2231.3   206.7 2225.49   247.1 2193.12   258.6 2189.37     325  2187.8
   338.8 2187.99   344.7 2189.62   359.2 2192.58   399.5 2192.21   416.1 2199.68
   421.9  2200.3   440.2 2195.47   498.1 2197.45   637.1 2196.11   659.5 2197.58
   677.5 2201.67   708.9 2201.33   722.3 2200.18   726.8 2201.28   749.5 2217.79
   762.7 2222.44   816.5 2229.41   852.3 2237.54   883.5 2249.46   943.8 2277.02
#Mann= 5 ,-1,0
       0      .1       0   258.6     .04       0   344.7      .1       0
   677.5    .016       0   708.9      .1       0
#XS Ineff= 2 , 0
                           447.5         2218.97
Permanent Ineff=
       F       F
#Block Obstruct= 1 ,-1
  544.84  578.09 2216.92
Bank Sta=258.6,344.7
XS Rating Curve= 0 ,0
Exp/Cntr(USF)=0,0
Exp/Cntr=0.5,0.3

Type RM Length L Ch R = 1 ,30034   ,495.6,483.5,443.2
XS GIS Cut Line= 3
2243954.75256414440262.252193784 2244371.8206863440382.424364576
2245029.23315004440396.562267022
#Sta/Elev= 30
       0 2303.51    59.8  2277.4    88.9 2266.74   101.4  2260.2   184.6 2232.73
     220 2225.47   242.7 2209.44   263.7 2190.43   269.92188.676   288.7 2187.01
   334.5 2186.94   351.1 2189.14   359.5 2190.88     372 2188.53   384.5 2190.79
   426.1 2191.15   456.7 2195.31   642.4 2193.72   710.5 2194.96   811.8  2194.2
   822.5 2194.84   836.4  2198.5   862.5 2198.17   870.5 2198.45   886.5 2209.77
   938.5 2242.41   958.5 2252.65   990.5 2266.47  1022.5 2276.08  1091.6 2291.58
#Mann= 6 ,-1,0
       0      .1       0   269.9     .04       0   351.1      .1       0
   456.7     .05       0   836.4    .016       0   862.5      .1       0
#XS Ineff= 2 , 0
                          833.58         2207.09
Permanent Ineff=
       F       F
Bank Sta=269.9,351.1
XS Rating Curve= 0 ,0
Exp/Cntr(USF)=0,0
Exp/Cntr=0.3,0.1

Type RM Length L Ch R = 1 ,29551   ,545.4,544.9,541.1
XS GIS Cut Line= 2
2243898.20095435440831.3027672392245050.44000371440820.699340404
#Sta/Elev= 30
       0 2303.26     110 2263.95     198 2243.03     210  2238.5     218 2237.43
     230 2231.18     250 2216.01     274 2192.61     282 2187.53     290 2186.41
     330 2186.38     370 2186.46   376.6 2187.56     386 2190.17   415.7 2190.65
     438 2195.53     530 2193.55     670 2193.16     742 2192.32     810    2194
     878 2193.94     882 2194.36     894 2199.47   920.4 2197.99     926 2198.44
     938 2206.25    1002  2240.7    1062 2265.87    1106 2278.82  1152.3    2287
#Mann= 6 ,-1,0
       0      .1       0     282     .04       0   376.6      .1       0
     670     .05       0     900    .016       0   920.4      .1       0
Bank Sta=282,376.6
XS Rating Curve= 0 ,0
Exp/Cntr(USF)=0,0
Exp/Cntr=0.3,0.1

Type RM Length L Ch R = 1 ,29006   ,476.6,476.5,476.9
Node Name=J
XS GIS Cut Line= 2
2243951.21808852441375.612011413 2245110.5260891441354.405157744
#Sta/Elev= 30
       0 2273.13      61  2247.6     113 2223.18     125 2215.64     145 2212.81
     165 2206.02     181 2190.82   186.52187.655     205 2185.32     265 2185.48
   271.5 2187.58     301 2189.09   309.8 2186.73  325.54 2186.72   368.7 2186.78
     377 2194.09     381 2194.28   520.1 2191.32   643.7 2192.86   777.1 2190.81
   869.1 2192.65   937.1 2191.35   953.1 2193.93   969.8 2203.57  1005.1 2203.28
  1009.1 2204.15  1037.1 2223.05  1066.2 2236.92  1113.1 2262.79  1159.5 2284.37
#Mann= 8 ,-1,0
       0      .1       0   186.5     .04       0   271.5      .1       0
  325.54     .04       0   368.7      .1       0   520.1     .05       0
   969.8    .016       0  1005.1      .1       0
Bank Sta=186.5,271.5
XS Rating Curve= 0 ,0
Exp/Cntr(USF)=0,0
Exp/Cntr=0.3,0.1

Type RM Length L Ch R = 1 ,28529   ,423.9,422.1,432
XS GIS Cut Line= 2
2243915.87333241441852.7662189682245198.88797939441828.024889688
#Sta/Elev= 30
       0 2283.32    20.3  2274.4   116.3 2226.48   164.3 2207.22   184.3 2201.47
   200.1 2199.72   207.9 2196.93   215.8  2192.8   222.1 2187.54   224.3 2185.62
   228.3    2185   248.3 2184.88   320.4 2184.97   329.6 2187.29   356.4 2187.48
   388.4 2191.44   464.4 2189.09   540.4 2191.43   620.4 2189.85   724.4 2190.02
   832.5 2192.07  1084.5 2191.05  1100.5 2193.27  1108.5 2198.24  1136.5 2200.74
    1143 2200.15  1148.5 2201.23  1160.5 2215.28  1208.5 2250.88  1283.3 2299.86
#Mann= 6 ,-1,0
       0      .1       0   222.1     .04       0   329.6      .1       0
     470     .05       0  1108.5    .016       0    1143      .1       0
Bank Sta=222.1,329.6
XS Rating Curve= 0 ,0
Exp/Cntr(USF)=0,0
Exp/Cntr=0.3,0.1

Type RM Length L Ch R = 1 ,28107   ,290.1,277.4,279.8
XS GIS Cut Line= 2
2243862.85619824442269.834341128  2245202.422455442269.834341128
#Sta/Elev= 30
       0 2296.77    57.3 2263.05   133.3 2223.77   169.3  2206.6   213.3 2191.41
   237.3 2187.61   249.3 2189.07   261.3 2188.32   274.32185.236   369.3 2184.44
   373.3 2184.96   409.3 2189.33   465.3 2189.78   513.3 2188.41   597.3 2190.94
   829.3 2188.73   949.3 2190.48   969.3  2191.9   981.3  2190.6  1141.3 2199.94
  1156.7  2202.3    1178 2203.62  1189.3 2203.05  1193.3 2202.23  1197.3 2204.08
  1209.3 2214.22    1254 2239.99  1297.3 2268.53  1309.3 2275.47  1339.6 2290.06
#Mann= 6 ,-1,0
       0      .1       0   274.3     .04       0   373.3      .1       0
     520     .05       0  1156.7    .016       0  1189.3      .1       0
Bank Sta=274.3,373.3
XS Rating Curve= 0 ,0
Exp/Cntr(USF)=0,0
Exp/Cntr=0.3,0.1

Type RM Length L Ch R = 1 ,27830   ,140.5,384.1,498.4
XS GIS Cut Line= 2
2243816.90801529442549.0579144382245117.59504033442541.988963215
#Sta/Elev= 30
       0  2279.4   103.3 2222.39   131.3  2204.2   152.2 2185.55   163.3 2182.98
   207.3 2184.45   243.3 2188.25   307.3 2186.93   319.3 2184.56   391.3 2184.51
   399.3 2188.22   451.3 2188.48   575.3 2188.34   671.5 2190.12   775.3 2186.78
   811.3    2189   907.3 2190.57   915.3 2189.57   927.3 2189.68  1087.3  2195.8
  1097.4 2197.09  1107.3 2201.67  1143.3 2202.58  1155.3  2200.6  1183.3 2201.44
  1203.3  2205.2  1227.3 2220.68  1239.3  2230.7  1258.2 2243.57  1300.7 2269.78
#Mann= 8 ,-1,0
       0      .1       0   319.3     .04       0   391.3      .1       0
   451.3     .05       0   915.3    .045       0   927.3     .05       0
  1107.3    .016       0  1143.3      .1       0
#Block Obstruct= 1 ,-1
    1034 1064.21 2214.81
Bank Sta=319.3,391.3
XS Rating Curve= 0 ,0
Exp/Cntr(USF)=0,0
Exp/Cntr=0.3,0.1

Type RM Length L Ch R = 1 ,27446   ,129.1,277.8,310.1
XS GIS Cut Line= 2
2243809.83906406442559.6613412732244541.47551565  443181.7290489
#Sta/Elev= 30
       0  2281.2    55.6 2249.63      68 2241.29    99.2 2215.93   134.3 2183.31
   156.7 2182.98   169.1  2185.1   223.6 2188.32   243.9 2186.74   267.9 2187.88
   348.9  2187.6   403.7 2185.27   480.9 2186.28   506.32183.833   516.4  2182.6
   601.6 2182.72   606.9 2183.85   612.1  2187.5   617.4 2188.02   681.6 2184.48
   712.5 2191.78   755.7 2194.58   768.1 2193.99   825.7  2215.1   842.2 2224.43
   866.9 2226.24   885.1 2237.56   913.6 2249.29   928.6  2253.2   960.3 2256.91
#Mann= 6 ,-1,0
       0      .1       0   506.3     .04       0   606.9     .06       0
     700    .016       0     760     .08       0     880      .1       0
#Block Obstruct= 2 ,-1
  836.55  872.87 2249.66  916.99  942.69 2275.31
Bank Sta=506.3,606.9
XS Rating Curve= 0 ,0
Exp/Cntr(USF)=0,0
Exp/Cntr=0.3,0.1

Type RM Length L Ch R = 1 ,27168   ,461.9,421.9,408.5
XS GIS Cut Line= 2
2243790.73421292442648.9198302532244126.67994654443275.403685809
#Sta/Elev= 30
       0 2266.21    27.5 2251.84    51.5 2237.51    70.8 2224.63      82 2215.73
    96.2 2196.57   104.6 2187.19   113.5 2183.15   138.5 2182.31   159.2 2185.85
   169.7 2185.15   181.8 2187.03   249.4 2186.72     259 2185.77   336.2 2187.29
   349.8  2186.5   352.8 2184.74   358.7 2182.38   364.7 2182.04     409 2181.78
   431.5 2182.25   438.5 2184.89   454.2 2191.98   488.7  2190.1   494.7 2191.43
   499.6 2194.85   522.3 2214.21   531.3 2217.33   576.7 2221.34   710.9 2239.33
#Mann= 5 ,-1,0
       0      .1       0   352.8     .04       0   438.5     .06       0
     460    .016       0   488.7      .1       0
Bank Sta=352.8,438.5
XS Rating Curve= 0 ,0
Exp/Cntr(USF)=0,0
Exp/Cntr=0.3,0.1

Type RM Length L Ch R = 1 ,26746   ,459,452.4,450.5
XS GIS Cut Line= 2
2243389.23646629442920.177853648 2243852.2527714 443506.90080516
#Sta/Elev= 30
       0 2376.93    56.9 2331.35    72.6 2319.75   101.6 2295.42     121 2275.13
   139.5 2253.38   153.3  2235.7   174.5 2212.67   194.9 2195.05     205 2188.23
   213.72184.135   220.4 2181.01   269.5 2180.51   288.8 2181.51   314.7 2183.84
   330.3 2182.68   359.9 2180.28   381.6 2180.79   398.7 2182.65   404.4 2184.28
   408.9 2186.08   430.9 2185.41   450.3 2188.11   470.1 2188.44   480.3 2188.77
   495.5  2197.7   510.8 2203.84   526.1 2208.29   551.6 2212.36   747.4 2231.78
#Mann= 8 ,-1,0
       0      .1       0   213.7     .04       0   288.8      .1       0
   330.3     .04       0   404.4      .1       0   450.3    .016       0
   470.1     .08       0   526.1      .1       0
Bank Sta=213.7,404.4
XS Rating Curve= 0 ,0
Exp/Cntr(USF)=0,0
Exp/Cntr=0.3,0.1

Type RM Length L Ch R = 1 ,26294   ,342.1,402.4,424.9
Node Name=I
XS GIS Cut Line= 2
2243031.82486816443204.0030517882243579.13506113443872.352998971
#Sta/Elev= 30
       0 2295.63      38 2287.59    55.1 2281.92    79.1 2270.71   110.1 2252.69
   123.3 2246.06   227.8 2200.57   245.5 2194.23   270.4 2188.33   280.7 2187.18
   296.92182.177   316.6 2179.25   341.5 2179.06   385.7  2179.3   401.9  2182.1
   430.3 2183.96   456.5 2182.92   477.2 2184.87   487.5 2183.02   495.7 2185.39
   537.2 2188.02   544.4 2189.31   555.4 2199.66   570.2  2208.4   580.9 2213.18
     598 2217.87   626.4 2221.94   663.5 2225.21   734.4 2234.96   863.9 2248.72
#Mann= 6 ,-1,0
       0      .1       0   296.9     .04       0   401.9      .1       0
   495.7    .016       0   537.2      .1       0     720     .05       0
Bank Sta=296.9,401.9
XS Rating Curve= 0 ,0
Exp/Cntr(USF)=0,0
Exp/Cntr=0.3,0.1

Type RM Length L Ch R = 1 ,25891   ,329.8,493.2,528.1
XS GIS Cut Line= 3
 2242869.6685514443224.1427562382242897.94435629443627.072975952
2243046.39233198443952.244732212
#Sta/Elev= 30
       0 2258.76     9.1 2254.96    49.2 2230.87    61.2 2225.07   109.3 2205.25
   145.4 2194.03   261.7 2188.03   325.6 2186.73   365.9 2187.74     374 2185.93
     386 2179.16     390 2178.62   406.2 2182.99   423.8 2180.15     437 2180.66
   445.8 2178.86     459  2179.8     4692178.371   494.2 2177.27   534.5 2178.32
     540  2180.7   573.3 2188.46     614 2191.57   626.1 2190.61   630.5 2191.35
   660.8 2211.92   669.3 2219.16   678.9 2223.64   722.8  2233.8   761.4 2240.15
#Mann= 5 ,-1,0
       0      .1       0     469     .04       0   534.5      .1       0
  583.92    .016       0  623.92      .1       0
#XS Ineff= 2 , 0
                           609.8         2199.95
Permanent Ineff=
       F       F
Bank Sta=469,534.5
XS Rating Curve= 0 ,0
Exp/Cntr(USF)=0,0
Exp/Cntr=0.3,0.1

Type RM Length L Ch R = 1 ,25398   ,367.9,491.1,514.3
XS GIS Cut Line= 2
2242743.32779189443195.7535938792242330.02179334443873.924659738
#Sta/Elev= 30
       0 2236.27    62.6 2212.68    95.4 2198.03   114.1 2192.22   123.5  2190.7
   184.4 2185.58   306.1 2186.69   385.8 2183.36   423.3 2183.53   451.6 2184.91
   483.82177.767     498 2176.66   540.4 2176.77   546.5 2177.61   559.1 2181.83
   568.5 2186.83   608.7 2190.36   626.2 2190.42   634.1  2192.9   646.6 2200.58
   657.5 2210.56   671.5 2220.65   675.7    2226   684.4 2233.23   713.2 2253.86
   718.4 2260.19   722.2 2263.33   733.9 2266.19   745.5 2272.67   794.2 2288.17
#Mann= 6 ,-1,0
       0      .1       0   483.8     .04       0   546.5      .1       0
     570    .016       0     630     .08       0     650      .1       0
Bank Sta=483.8,546.5
XS Rating Curve= 0 ,0
Exp/Cntr(USF)=0,0
Exp/Cntr=0.3,0.1

Type RM Length L Ch R = 1 ,24907   ,506,501.3,500.5
XS GIS Cut Line= 2
2242671.37954215443074.3226855852241981.97920293 443342.71518406
#Sta/Elev= 30
       0 2248.41    38.7 2239.93    97.4 2231.45     119 2226.08   143.7 2217.88
   173.3 2205.18   183.9 2202.25   227.1  2185.8   242.6 2184.24   298.2 2183.03
   338.6 2185.28     364 2184.94   415.5 2180.65   483.6 2181.41   493.12177.672
   497.1  2175.8   501.4 2175.29   561.5 2175.36   570.2  2177.4   582.4 2183.31
   587.2 2184.62     613 2185.59   621.6 2184.81   625.7 2186.16   638.1 2197.29
   651.6 2210.85   668.8 2225.57   681.6 2238.19   690.2 2242.36   739.8 2256.59
#Mann= 5 ,-1,0
       0      .1       0   493.1     .04       0   570.2      .1       0
     580    .016       0     620      .1       0
Bank Sta=493.1,570.2
XS Rating Curve= 0 ,0
Exp/Cntr(USF)=0,0
Exp/Cntr=0.3,0.1

Type RM Length L Ch R = 1 ,24406   ,499.5,498,497.2
XS GIS Cut Line= 2
2242321.82483161442662.161134007 2241766.9121606442895.436524367
#Sta/Elev= 30
       0 2233.84    36.5 2226.15    98.3  2204.2   127.6 2191.29   144.1 2186.91
   166.7 2184.92   186.9 2180.26     197 2179.31   227.4 2179.91   236.1  2178.8
   249.1 2180.57   270.8 2180.33   279.5 2179.79   285.22176.714   292.5 2173.32
   301.2 2172.48   396.6 2173.43     401 2173.77   407.52176.716     419 2181.39
   454.1 2182.63   461.8 2183.38   479.1 2198.51   492.1 2204.85   505.1 2215.13
   539.8 2237.24   544.2 2239.05   552.9  2239.6   565.9 2247.73     602 2264.95
#Mann= 5 ,-1,0
       0      .1       0   285.2     .04       0   407.5      .1       0
     420    .016       0   454.1      .1       0
Bank Sta=285.2,407.5
XS Rating Curve= 0 ,0
Exp/Cntr(USF)=0,0
Exp/Cntr=0.3,0.1

Type RM Length L Ch R = 1 ,23908   ,362.7,360.4,358.6
XS GIS Cut Line= 2
2242170.72865393 442180.235684162241528.69169679442459.153378654
#Sta/Elev= 30
       0 2273.56    24.6    2270    52.6 2264.83   112.1 2248.51   120.5 2245.33
   151.6 2230.15   242.6 2192.02   290.6 2179.25   313.6 2177.34     331 2177.57
   334.1 2177.09   340.32174.115   346.2 2171.74   349.3 2171.38   403.9 2171.25
   425.3 2171.42     434  2174.2   443.3 2179.01   446.5 2179.36     477 2180.36
   492.2 2179.78     500 2178.47   504.3 2178.63   507.4 2180.33   521.8 2190.88
   556.7 2220.11   569.7 2232.16   586.4 2245.24   635.2 2273.52     700 2313.19
#Mann= 6 ,-1,0
       0     .12       0      70      .1       0   340.3     .04       0
     434      .1       0     460    .016       0     500      .1       0
Bank Sta=340.3,434
XS Rating Curve= 0 ,0
Exp/Cntr(USF)=0,0
Exp/Cntr=0.3,0.1

Type RM Length L Ch R = 1 ,23547   ,358.8,357.4,365.5
Node Name=H
XS GIS Cut Line= 2
2241975.44622168441863.3696458032241402.86117262442128.455316667
#Sta/Elev= 30
       0 2250.15    21.2 2245.96      52 2242.64    74.1 2239.26   113.8 2228.73
   127.4 2223.81   137.6    2219   171.1 2200.35     202 2190.63   237.2 2175.56
   254.9 2175.88   286.12173.984   298.9 2171.53   308.1 2171.04   382.7 2171.12
   394.7 2173.71   404.6  2175.7   413.6 2180.41   422.4 2180.85   448.8 2178.83
   453.2 2179.58   461.8 2186.29   470.8 2194.75   484.1 2209.17   492.9 2215.78
   497.3 2218.02   506.1 2219.49   519.3 2228.22   603.1 2269.31     631 2284.87
#Mann= 5 ,-1,0
       0      .1       0   286.1     .04       0   394.7     .08       0
   413.6    .016       0     450      .1       0
Bank Sta=286.1,394.7
XS Rating Curve= 0 ,0
Exp/Cntr(USF)=0,0
Exp/Cntr=0.3,0.1

Type RM Length L Ch R = 1 ,23190   ,498.2,427.7,206.8
XS GIS Cut Line= 3
2241858.66371061441515.9678282992241268.55109938441803.283560407
2241220.23945991441932.417148379
#Sta/Elev= 30
       0 2230.69    17.7 2229.28    42.8 2224.95    82.8 2223.97   103.3 2221.87
   128.4 2222.11   140.7 2220.33   162.9 2213.07   185.5 2201.99   206.2 2194.49
   233.2 2178.75     243 2175.52   272.1 2172.02   323.1 2176.81   368.8 2171.51
   388.8 2170.66   469.9 2171.46   478.8 2176.45   483.3  2177.2   527.7 2178.89
   560.2 2177.51   578.4 2182.05   587.6 2182.24   628.1 2178.85   633.3  2180.5
   646.1 2188.33   656.3 2191.41   670.5 2202.15   739.5 2247.41   794.2 2286.93
#Mann= 7 ,-1,0
       0      .1       0   368.8     .04       0   469.9      .1       0
     500     .05       0   587.6    .016       0     650     .08       0
  706.34      .1       0
#XS Ineff= 2 , 0
                          582.76         2197.46
Permanent Ineff=
       F       F
Bank Sta=368.8,469.9
XS Rating Curve= 0 ,0
Exp/Cntr(USF)=0,0
Exp/Cntr=0.3,0.1

Type RM Length L Ch R = 1 ,22762   ,339,324.3,228.5
XS GIS Cut Line= 2
  2241335.706136441142.3366210532241134.24102614 441902.24887753
#Sta/Elev= 30
       0 2219.54    70.6 2205.05   102.3 2203.39   110.5 2201.96   118.8 2196.09
   127.1 2186.79   139.3 2176.52   143.6 2173.15   150.72170.338   160.2 2168.72
   237.5 2168.51   247.1 2168.69   252.4  2169.9   259.5 2171.57   288.5 2174.37
     334 2175.22   354.7 2173.02   397.7  2176.8     483 2178.19   545.2 2176.32
   582.3 2177.49   598.8 2181.25   610.3 2181.13   631.9 2179.03   636.1 2179.86
   652.2 2194.16   681.6 2213.63   741.2 2255.52   772.6 2275.85   786.2 2286.54
#Mann= 7 ,-1,0
       0      .1       0   150.7     .04       0   252.4      .1       0
   397.7     .06       0   610.3    .016       0   652.2     .08       0
   741.2      .1       0
#XS Ineff= 2 , 0
                          599.44         2201.33
Permanent Ineff=
       F       F
Bank Sta=150.7,252.4
XS Rating Curve= 0 ,0
Exp/Cntr(USF)=0,0
Exp/Cntr=0.3,0.1

Type RM Length L Ch R = 1 ,22438   ,262.8,243.7,118
XS GIS Cut Line= 2
2240970.61258893441147.5977054582240969.40003783441911.504898441
#Sta/Elev= 30
       0 2224.44    33.6 2217.11    73.6 2211.22    93.6 2205.87   113.6 2197.83
   129.6  2187.8   141.6 2181.92     1852169.436   189.6 2167.64   213.6 2167.17
   237.6 2167.49   247.5  2168.9   289.6 2171.09   301.6 2170.77   307.6 2169.23
   313.6 2167.81   353.6 2167.88   363.4 2170.51   369.6  2174.4   389.6 2175.37
   449.6 2176.73   511.2 2174.59   541.6 2175.28   557.6 2180.51   573.6 2180.89
   597.6 2178.49   601.6 2179.49   620.1 2192.98   696.2 2229.22   763.9 2259.39
#Mann= 8 ,-1,0
       0      .1       0     185     .04       0   247.5      .1       0
   307.6     .04       0   363.4      .1       0   511.2     .08       0
   573.6    .016       0   620.1      .1       0
Bank Sta=185,363.4
XS Rating Curve= 0 ,0
Exp/Cntr(USF)=0,0
Exp/Cntr=0.3,0.1

Type RM Length L Ch R = 1 ,22194   ,613,590.8,512.2
XS GIS Cut Line= 2
2240639.41444053441202.4227064482240964.58619679441923.455731199
#Sta/Elev= 30
       0 2252.38      45 2240.91   108.5 2227.66   121.5 2223.24   125.9 2220.74
   139.1  2211.1   169.8 2182.48   187.3 2170.16   191.7 2167.82   199.2 2166.54
   235.6 2166.44   244.4 2166.99   253.1 2167.13   327.7 2167.17   332.1 2167.25
   337.32168.591   349.7 2173.67   358.4 2174.18     455 2174.91   490.1 2174.05
   559.1 2176.45   580.3 2180.82   586.3 2181.28   617.3 2178.69   621.7 2181.22
   630.5 2188.88   639.3  2195.4   737.5 2236.72   766.5 2250.45     791 2263.33
#Mann= 8 ,-1,0
       0      .1       0   191.7     .04       0   244.4      .1       0
   253.1     .04       0   337.3      .1       0   490.1     .08       0
   580.3    .016       0   630.5      .1       0
Bank Sta=191.7,337.3
XS Rating Curve= 0 ,0
Exp/Cntr(USF)=0,0
Exp/Cntr=0.3,0.1

Type RM Length L Ch R = 1 ,21603   ,554.5,555.7,559.3
XS GIS Cut Line= 2
2240084.50176952441598.2839749392240639.41444053442103.713987386
#Sta/Elev= 30
       0 2303.92    53.7 2262.37    69.6 2249.04   129.2 2207.45   177.4 2180.45
   183.5 2176.22   191.5 2169.34   194.3 2167.88   202.72165.971   210.6  2163.9
   228.3 2163.42   290.6 2163.62     308 2165.91   318.8 2167.32     331 2170.52
   340.4  2171.2   364.3 2171.82   395.4 2170.69   460.5 2172.71   515.2 2175.78
   521.1 2176.74   528.5 2180.46     537  2182.1   562.7 2180.88   567.7 2182.69
   576.6 2187.38   610.2 2197.56   661.6 2212.54   689.9 2218.91   750.6 2237.69
#Mann= 6 ,-1,0
       0      .1       0   202.7     .04       0     308      .1       0
   528.5    .016       0     570     .08       0   610.2      .1       0
#Block Obstruct= 1 ,-1
  687.54  743.76 2255.35
Bank Sta=202.7,308
XS Rating Curve= 0 ,0
Exp/Cntr(USF)=0,0
Exp/Cntr=0.3,0.1

Type RM Length L Ch R = 1 ,21048   ,467,491.7,508.3
XS GIS Cut Line= 2
2239660.36469614441951.7315360912240225.88079398442492.506304654
#Sta/Elev= 30
       0 2314.39    48.4  2279.1    54.2 2276.18   123.6 2227.86   187.6 2191.08
   216.2 2178.72   227.8 2174.91   239.4 2172.46   275.3 2169.85   279.9 2168.76
   288.62164.326   293.1  2162.7   303.6 2161.69   372.5 2161.59   392.7 2161.83
   401.4 2164.11   424.6 2167.78   447.7 2169.62   503.4 2172.08     520 2177.28
   552.6 2177.85   563.5 2183.22   580.9 2185.59   600.7 2192.03   640.3  2200.9
   679.3 2217.74   690.8 2224.41   702.4  2228.6   724.8 2241.39   782.5  2277.3
#Mann= 7 ,-1,0
       0      .1       0   288.6     .04       0   401.4      .1       0
     520    .016       0     550     .06       0   563.5     .03       0
   580.9      .1       0
Bank Sta=288.6,401.4
XS Rating Curve= 0 ,0
Exp/Cntr(USF)=0,0
Exp/Cntr=0.3,0.1

Type RM Length L Ch R = 1 ,20556   ,494,539.3,554.9
Node Name=G
XS GIS Cut Line= 2
2239276.84736451442136.0868099762239739.95598933442788.648963132
#Sta/Elev= 30
       0 2328.73    11.1 2320.36    40.5 2300.64    60.2 2285.85      70  2277.3
   109.2 2250.32   123.2 2241.64   157.8 2222.02   231.9  2187.5   258.5 2178.05
     276 2174.38   325.1 2169.69   388.8 2169.77   419.2 2163.89   431.42162.467
   439.2  2160.2   470.8 2159.94   506.5  2160.2     511 2160.77   513.8 2162.32
   521.3 2165.72   545.8 2170.16   579.4 2171.57     597 2182.39   614.5 2190.85
   660.2  2216.6   712.6 2248.71     742 2268.71   761.6 2284.23   800.2 2311.94
#Mann= 6 ,-1,0
       0      .1       0   431.4     .04       0   513.8     .03       0
     550    .016       0     570     .08       0   579.4      .1       0
#XS Ineff= 2 , 0
                          564.51         2187.24
Permanent Ineff=
       F       F
Bank Sta=431.4,513.8
XS Rating Curve= 0 ,0
Exp/Cntr(USF)=0,0
Exp/Cntr=0.3,0.1

Type RM Length L Ch R = 1 ,20017   ,447.5,454.5,457
XS GIS Cut Line= 2
2238918.12481772442347.5928045812239176.14153736443047.418975662
#Sta/Elev= 30
       0 2264.79    30.9 2251.33    44.3 2244.22   108.3 2200.84   142.4 2188.39
   172.2 2181.55   230.2 2172.43   261.7 2169.18   321.4 2167.93   339.2 2164.27
   363.9 2167.53   379.7  2166.9   398.2 2163.62   407.22160.635   444.9 2159.41
     480 2160.36   496.2 2169.81   526.3 2171.88   530.3 2171.43   535.5 2173.13
   549.4 2185.78     553 2191.06   560.4 2204.65   564.4 2209.59   611.3 2242.74
   632.6 2263.02   658.2 2283.53   679.5 2299.18   739.2 2338.35   745.9 2343.88
#Mann= 5 ,-1,0
       0      .1       0   407.2     .04       0     480      .1       0
     500    .016       0   526.3      .1       0
#XS Ineff= 2 , 0
                          515.15         2184.17
Permanent Ineff=
       F       F
Bank Sta=407.2,480
XS Rating Curve= 0 ,0
Exp/Cntr(USF)=0,0
Exp/Cntr=0.3,0.1

Type RM Length L Ch R = 1 ,19562   ,473.1,482.8,477.6
XS GIS Cut Line= 2
2238508.12564678442481.902877819 2238727.2631347443185.263524512
#Sta/Elev= 30
       0 2302.22    12.2 2293.07    24.4 2285.66    45.3 2269.18    57.9 2261.85
    95.3 2233.88   116.6 2219.43   137.5 2203.76   166.8 2185.75   196.2 2169.71
   204.5 2168.19   254.8 2166.98   309.5 2166.13   334.4  2167.2   366.8 2160.74
   372.1 2159.99   456.3 2159.88   464.3 2160.78   476.9 2168.42   481.8 2170.28
   510.4  2171.5   514.6 2172.33   518.8 2175.11   539.7 2194.39   574.5 2215.98
   612.8 2241.37   635.1 2257.52   679.9 2287.72   692.6 2298.07   736.7 2328.04
#Mann= 5 ,-1,0
       0      .1       0   366.8     .04       0   464.3      .1       0
   481.8    .016       0   510.4      .1       0
#XS Ineff= 2 , 0
                          485.86         2186.98
Permanent Ineff=
       F       F
Bank Sta=366.8,464.3
XS Rating Curve= 0 ,0
Exp/Cntr(USF)=0,0
Exp/Cntr=0.3,0.1

Type RM Length L Ch R = 1 ,19079   ,463.4,483,477.4
XS GIS Cut Line= 2
2238055.71276851442598.540572999 2238267.7813052443330.177024584
#Sta/Elev= 30
       0 2315.39     6.9  2310.1    27.7    2288    48.6 2273.11   102.2 2230.74
   127.7 2212.57   144.3 2203.28     161 2191.23   190.2 2176.89   218.8 2166.53
   256.8 2165.49   265.1 2163.71   277.6 2163.99   284.52161.325   290.1 2159.12
   306.8 2158.59   444.2 2159.12   451.8 2161.59     465 2168.68   480.4 2170.43
   506.7 2169.75   510.8 2170.18   519.3 2175.53     540 2184.59   593.4 2211.15
   648.3 2239.95   698.2 2269.48   706.6 2277.93   710.7 2280.15   761.8 2298.18
#Mann= 5 ,-1,0
       0      .1       0   284.5     .04       0   451.8      .1       0
   480.4    .016       0   506.7      .1       0
#XS Ineff= 2 , 0
                           480.9          2180.7
Permanent Ineff=
       F       F
Bank Sta=284.5,451.8
XS Rating Curve= 0 ,0
Exp/Cntr(USF)=0,0
Exp/Cntr=0.3,0.1

Type RM Length L Ch R = 1 ,18596   ,403.7,411.6,432.9
XS GIS Cut Line= 2
2237628.04121951442743.4540730722237787.09262203443450.349195376
#Sta/Elev= 30
       0 2260.68    38.4 2238.18    51.8  2231.5    96.1 2204.63   115.4 2194.25
   142.1 2181.59   161.7 2174.33   178.1 2166.32   198.3 2158.97   208.4 2157.44
   321.6 2158.63   328.6 2159.48     338 2161.28   342.1 2161.04   349.6 2158.67
   383.1 2158.03   396.5 2158.85   415.9 2170.38   432.3 2171.67   451.8 2170.91
   456.9 2172.14   465.1  2178.6   470.1 2181.28   493.8 2191.05     527 2207.01
   563.8 2222.42   596.3 2234.56   653.7 2253.87   711.3 2275.43   724.6 2281.22
#Mann= 7 ,-1,0
       0      .1       0   198.3     .04       0   328.6      .1       0
   349.6     .04       0   396.5      .1       0   415.9    .016       0
   451.8      .1       0
#XS Ineff= 2 , 0
                          422.76         2183.42
Permanent Ineff=
       F       F
Bank Sta=198.3,396.5
XS Rating Curve= 0 ,0
Exp/Cntr(USF)=0,0
Exp/Cntr=0.3,0.1

Type RM Length L Ch R = 1 ,18185   ,327,332.1,357.2
XS GIS Cut Line= 2
2237249.85232908442792.936731633 2237317.0073657443485.693951491
#Sta/Elev= 30
       0 2287.96    12.3 2274.16    28.4  2263.3    44.4 2248.16    52.5 2244.15
    64.5 2234.22    72.6  2230.2   120.8 2196.39   141.6 2185.23     161 2169.53
     173 2165.91   180.62159.805   189.1 2157.03   229.1 2156.88   253.4 2157.07
   260.2 2160.29   265.5 2163.04   273.5 2164.31   305.7 2159.93   349.2 2159.43
   361.9 2157.03   406.1 2157.01   414.2 2159.16   430.2 2171.31   438.3  2175.1
   466.4 2175.35   490.5 2196.67   632.5 2282.83   647.4 2293.73     696 2319.77
#Mann= 7 ,-1,0
       0      .1       0   180.6     .04       0   260.2      .1       0
   349.2     .04       0   414.2      .1       0   430.2    .016       0
   466.4      .1       0
Bank Sta=180.6,414.2
XS Rating Curve= 0 ,0
Exp/Cntr(USF)=0,0
Exp/Cntr=0.3,0.1

Type RM Length L Ch R = 1 ,17853   ,129.2,132.2,216
Node Name=F
XS GIS Cut Line= 2
2236945.88742649442764.6609267412236928.21504843443471.556049045
#Sta/Elev= 30
       0 2296.28    12.5 2286.25    64.5 2254.41     126  2210.5   136.6 2205.41
   158.8 2189.89   224.5  2158.9   232.7 2156.16   268.6  2156.1   280.6 2156.64
   287.1 2159.44   292.6 2160.51   332.6 2160.65   361.3 2158.97   372.6  2157.5
   384.6 2157.69   408.6 2155.96   452.7 2155.99   456.7 2156.24   460.7 2158.65
   476.7 2170.56   480.7 2172.95   484.7 2173.93   508.7 2175.76   515.9 2175.27
   520.7 2176.23   536.7 2191.36   564.7 2212.37   584.7 2226.25   707.1  2300.8
#Mann= 7 ,-1,0
       0      .1       0   224.5     .04       0   287.1      .1       0
   361.3     .04       0   460.7      .1       0   484.7    .016       0
   515.9      .1       0
Bank Sta=224.5,460.7
XS Rating Curve= 0 ,0
Exp/Cntr(USF)=0,0
Exp/Cntr=0.3,0.1

Type RM Length L Ch R = 1 ,17720   ,361.3,364,306.7
XS GIS Cut Line= 4
2236829.24973131442764.6609267412236800.97392642443093.367158612
2236726.74993858443167.5911464542236684.33623124443453.883670987
#Sta/Elev= 30
       0 2278.63    49.5 2250.64    72.8 2239.62   169.1 2181.44   185.2 2174.05
   197.4 2171.01   212.22158.154   221.3 2155.52   269.5 2155.62   273.5 2155.72
   280.5 2158.84   289.6 2161.03   313.7 2161.66   352.3  2159.3   361.5 2155.85
   393.3  2155.3   404.6 2156.37   460.8 2155.37   476.9 2157.55     485 2161.15
   494.9 2168.05   505.2 2171.47   533.4 2172.87   545.7 2182.81   569.9  2210.3
     578 2217.13   614.4 2244.47   622.5  2252.8   699.5 2310.99   724.3 2328.35
#Mann= 7 ,-1,0
       0      .1       0   212.2     .04       0   280.5      .1       0
   352.3     .04       0   476.9      .1       0   494.9    .016       0
   533.4      .1       0
Bank Sta=212.2,476.9
XS Rating Curve= 0 ,0
Exp/Cntr(USF)=0,0
Exp/Cntr=0.3,0.1

Type RM Length L Ch R = 1 ,17356   ,466.1,462.2,461.3
XS GIS Cut Line= 2
2236482.44418872442724.5123381132236387.01334721443374.855850633
#Sta/Elev= 30
       0 2265.88    44.9 2239.33    73.4 2225.02    97.7 2209.72   109.8 2204.38
     122 2196.08   154.3 2179.74   178.6 2170.06   206.7 2155.59   231.1 2154.63
   267.5 2154.83   275.6 2156.96   287.7 2159.46   303.9 2158.16   344.3 2158.55
   356.4 2156.78   372.6 2159.25   383.3 2157.51   390.4 2155.59  426.38 2155.39
   441.3 2166.06   453.5 2168.93   477.7  2169.3   485.6 2175.11   493.9 2187.95
   497.9 2192.18   554.5 2235.49   631.4 2286.05   649.3 2296.66   657.3 2298.86
#Mann= 7 ,-1,0
       0      .1       0   206.7     .04       0   275.6      .1       0
   383.3     .04       0  426.38      .1       0   441.3    .016       0
   477.7      .1       0
Bank Sta=206.7,426.38
XS Rating Curve= 0 ,0
Exp/Cntr(USF)=0,0
Exp/Cntr=0.3,0.1

Type RM Length L Ch R = 1 ,16894   ,293.9,306.6,303
XS GIS Cut Line= 3
2236005.71691383 442648.023231562235988.04453577442962.591560986
2235917.35502354443316.039122138
#Sta/Elev= 30
       0 2196.74    37.2 2193.37    85.3 2194.23   149.4 2185.91   165.4 2180.21
   177.4 2173.96   205.72155.255   209.5 2153.26   217.5 2152.93   269.6 2153.06
   288.2 2155.78   321.8 2158.49   346.3 2156.45   354.5 2153.47   369.9  2154.2
   389.9 2162.85   403.4 2164.09   427.8 2163.02   444.2 2177.63   468.6 2202.68
   501.3 2228.18   514.3 2239.75   538.8 2255.38   562.5 2281.48   582.9 2298.25
     591 2310.95   606.1 2331.18   631.8 2352.79     640 2361.77   675.5 2382.54
#Mann= 7 ,-1,0
       0      .1       0   205.7     .04       0   288.2      .1       0
   346.3     .04       0   369.9      .1       0   389.9    .016       0
   427.8      .1       0
#XS Ineff= 2 , 0
                           399.1         2182.66
Permanent Ineff=
       F       F
Bank Sta=205.7,369.9
XS Rating Curve= 0 ,0
Exp/Cntr(USF)=0,0
Exp/Cntr=0.3,0.1

Type RM Length L Ch R = 1 ,16588   ,340.5,340.2,341
XS GIS Cut Line= 2
2235756.09106547442485.3028626212235629.78871324   443264.167368
#Sta/Elev= 30
       0 2238.23   113.3 2201.05   178.2 2191.56   218.7 2184.04   299.8 2173.32
     320 2168.04   336.2 2161.97   376.4 2159.11   384.8 2157.39   390.42154.778
     397 2152.45   404.3 2152.12   467.1 2152.31   477.5 2155.58   486.1 2160.57
   494.2 2162.64   518.6 2163.66   530.7 2162.43   534.8 2164.11   550.7 2179.96
   556.2 2184.09   579.3 2198.92   587.5 2201.94   636.1 2234.01   648.2 2248.12
   684.7 2273.05   692.8 2283.81   696.4 2286.25     746 2310.99     789 2337.59
#Mann= 6 ,-1,0
       0      .1       0   390.4     .04       0   477.5     .08       0
     490    .016       0     540     .08       0   556.2      .1       0
#XS Ineff= 2 , 0
                          503.89         2174.87
Permanent Ineff=
       F       F
Bank Sta=390.4,477.5
XS Rating Curve= 0 ,0
Exp/Cntr(USF)=0,0
Exp/Cntr=0.3,0.1

Type RM Length L Ch R = 1 ,16248   ,384.5,373.4,368.5
XS GIS Cut Line= 2
2235429.59738915442386.472036308 2235291.7528403443217.073805015
#Sta/Elev= 30
       0 2288.91    31.1 2270.17    39.2 2263.38    55.5 2252.41   108.2 2222.78
   152.8  2202.9   198.3 2184.84   221.7 2176.97     253 2169.45   339.3 2162.96
   347.4 2161.29   359.6 2160.64   379.8 2155.34     392 2155.94   400.1 2157.56
   408.42154.394   416.3 2152.64   497.4 2152.25   501.5 2152.32   507.2 2154.27
   521.7 2162.81   529.9 2165.45   562.3 2164.92   586.6  2186.4   619.1 2206.34
   668.4 2237.48   752.9 2294.61   773.1 2305.79   809.6 2331.12     842 2348.79
#Mann= 6 ,-1,0
       0      .1       0   408.4     .04       0   507.2     .08       0
     530    .016       0     570     .08       0   619.1      .1       0
#XS Ineff= 2 , 0
                           536.9         2175.88
Permanent Ineff=
       F       F
Bank Sta=408.4,507.2
XS Rating Curve= 0 ,0
Exp/Cntr(USF)=0,0
Exp/Cntr=0.3,0.1

Type RM Length L Ch R = 1 ,15874   ,589.4,609.8,598.4
XS GIS Cut Line= 2
2235023.13269382442305.179097243 2234955.9776572443160.522195231
#Sta/Elev= 30
       0  2274.8    18.6 2267.39    72.2 2243.46    88.3 2238.06   172.5  2202.7
   218.8 2185.32   268.8 2170.89     313 2163.65     333 2159.55     341 2159.08
   361.1 2152.33   373.1 2151.16   385.2 2154.28   405.2 2151.78     4262152.893
   516.1 2153.27   541.7 2165.01   549.7 2166.28   561.7 2173.16   573.8 2174.01
   593.8 2173.49     598 2174.39   609.9 2181.53   629.9 2199.46   633.9 2202.28
   683.6 2231.81   746.3 2270.61   758.3  2280.2     810 2312.95     858 2340.57
#Mann= 7 ,-1,0
       0      .1       0     426     .04       0   516.1      .1       0
     530     .04       0     560    .016       0     600     .08       0
     630      .1       0
Bank Sta=426,516.1
XS Rating Curve= 0 ,0
Exp/Cntr(USF)=0,0
Exp/Cntr=0.3,0.1

Type RM Length L Ch R = 1 ,15264   ,858.1,848.7,826.9
XS GIS Cut Line= 2
 2234464.6855472442220.351682566 2234340.9789008443089.832683001
#Sta/Elev= 30
       0 2375.62    33.2 2352.09    61.6 2329.41    69.5 2322.19    85.7  2302.8
     122 2275.47   259.2 2189.47   287.7 2166.93   315.82152.265   332.1 2149.92
   412.9 2149.97     421 2151.68   425.1 2154.58   432.7 2155.41   476.1 2159.74
   545.9  2158.1   562.4 2161.76   574.6 2169.23   590.7  2183.2   602.5 2185.51
     623 2184.54   630.8 2188.28   639.2 2202.02   643.2 2205.58   651.3 2208.74
   671.5 2222.09     720 2244.67     787 2276.42     853 2303.55   878.2  2316.6
#Mann= 9 ,-1,0
       0      .1       0   315.8     .04       0     421     .07       0
   432.7      .1       0   476.1     .06       0   545.9      .1       0
   602.5    .016       0   630.8     .08       0     720      .1       0
Bank Sta=315.8,421
XS Rating Curve= 0 ,0
Exp/Cntr(USF)=0,0
Exp/Cntr=0.3,0.1

Type RM Length L Ch R = 1 ,14416   ,628.1,639.4,619.9
Node Name=E
XS GIS Cut Line= 2
2233571.33762789442152.1875272682233560.81243187443041.566590843
#Sta/Elev= 30
       0  2257.9      69 2231.86     133 2211.83     157 2202.23     193 2190.16
     265 2170.97   277.1 2165.31     293 2160.46     3042153.674     313 2150.87
     353 2149.78     413 2149.96     417 2150.61     421 2153.23     425 2155.39
     441 2156.75     521 2155.67     565 2159.07     649 2177.57     661 2181.96
     673 2191.01     685 2194.59     713 2193.61     717 2193.45     737  2208.7
   783.2 2233.47   837.1 2265.59   849.1 2267.65   865.1 2280.52   889.4 2293.17
#Mann= 5 ,-1,0
       0      .1       0     304     .04       0     421      .1       0
     673    .016       0     713      .1       0
Bank Sta=304,421
XS Rating Curve= 0 ,0
Exp/Cntr(USF)=0,0
Exp/Cntr=0.3,0.1

Type RM Length L Ch R = 1 ,13776   ,658.3,657.2,651.1
XS GIS Cut Line= 2
2232938.56008482442111.7366347752232949.08528084 442995.85310034
#Sta/Elev= 30
       0  2285.8    48.4 2279.44    69.4 2274.99   101.9 2265.69   137.5  2251.1
   197.5 2213.35   226.5 2190.58   257.5 2169.84   269.5 2163.28   281.5  2159.4
   298.62151.229   305.5 2149.56   380.92150.689   453.5 2151.28   465.5 2148.78
   501.5 2156.45   529.5 2154.98   576.2 2156.29   637.5 2155.42   661.5 2157.69
   693.5 2167.05   725.5  2179.1   744.7 2193.62   750.2 2195.58   773.5 2195.56
   777.5 2195.65   781.5 2198.07   797.5 2213.97   805.5 2219.52   884.2 2267.71
#Mann= 6 ,-1,0
       0      .1       0   298.6     .04       0   380.9      .1       0
     630     .05       0   750.2    .016       0   773.5      .1       0
Bank Sta=298.6,380.9
XS Rating Curve= 0 ,0
Exp/Cntr(USF)=0,0
Exp/Cntr=0.3,0.1

Type RM Length L Ch R = 1 ,13119   ,1164.2,1115.9,637.5
XS GIS Cut Line= 2
2232273.26818391442124.0681840072232310.10636997443087.123619712
#Sta/Elev= 30
       0 2340.24     9.1 2338.61    37.1 2315.69    53.1 2309.58    65.2 2298.52
   101.2 2270.85   161.2 2228.52   209.3 2196.99   221.3 2186.93   237.3 2179.63
   273.3 2156.23   281.3 2152.67   289.2 2151.85   349.4 2147.62   361.4 2147.74
   377.9 2151.26   405.4 2154.54   445.4 2154.76   561.5 2154.53   713.6 2151.06
   745.7 2152.27   769.7 2160.14   797.3 2173.56   825.7 2194.49   837.7 2200.15
   861.7    2199   869.7 2202.93   889.8 2219.34   898.3 2228.73   963.8  2269.1
#Mann= 6 ,-1,0
       0      .1       0   289.2     .04       0   377.9      .1       0
   445.4     .05       0   837.7    .016       0   861.7      .1       0
Bank Sta=289.2,377.9
XS Rating Curve= 0 ,0
Exp/Cntr(USF)=0,0
Exp/Cntr=0.3,0.1

Type RM Length L Ch R = 1 ,12003   ,968.8,915.9,355.6
Node Name=D
XS GIS Cut Line= 2
2231020.14401116442500.5430409382231988.46204487443195.205978168
#Sta/Elev= 30
       0 2285.53    14.8 2273.63    62.9 2241.96    72.1 2232.41    83.6 2229.53
    89.3 2225.95   132.3 2189.36   172.6 2156.93   179.5 2153.46   189.7 2151.86
   198.3 2146.92   206.8 2145.41   278.82146.373   295.4 2148.28   304.3 2147.39
   315.1 2145.55   330.1 2145.84   334.8 2147.34   339.7 2150.81   344.6  2152.3
   460.9 2151.01   542.2    2152   654.8 2150.28    1051  2150.2  1066.8 2154.18
  1081.1 2162.74  1097.8 2175.57  1118.4 2184.34  1164.3 2192.27  1191.7 2203.34
#Mann= 7 ,-1,0
       0      .1       0   198.3     .04       0   278.8      .1       0
   304.3    .045       0   334.8     .01       0   460.9     .05       0
  1081.1     .08       0
#Block Obstruct= 1 ,-1
 1108.06 1130.49 2206.44
Bank Sta=198.3,278.8
XS Rating Curve= 0 ,0
Exp/Cntr(USF)=0,0
Exp/Cntr=0.3,0.1

Type RM Length L Ch R = 1 ,11087   ,505.7,498.1,435
XS GIS Cut Line= 3
2231156.41637482443616.4695491172231792.62198489443224.142756238
2231994.08709475443217.073805015
#Sta/Elev= 30
       0 2178.86    31.3 2186.09    60.8 2195.48    84.3 2196.21     101 2190.06
   115.6 2181.77   148.5 2151.13   162.92144.863   173.6 2142.69   227.3 2142.59
   246.4  2142.8   257.8 2145.11   269.6 2149.37   298.7 2148.99     324 2146.63
   394.5 2148.87   648.2  2148.6   676.6    2150   723.4 2158.02   732.8 2161.39
   746.4 2161.03     759 2167.12     803 2170.83     819 2176.23   839.3 2179.79
   875.1 2182.22   891.1  2187.9   916.2 2191.65   939.1 2201.89     949  2202.5
#Mann= 8 ,-1,0
       0     .12       0      40      .1       0   162.9     .04       0
   257.8      .1       0   298.7     .05       0     730    .016       0
   746.4     .05       0     949     .03       0
#Block Obstruct= 5 ,-1
  629.58  684.75 2171.27  697.68  718.94 2177.47  756.12  804.12 2191.18
  840.95  868.02 2201.85  888.93  913.83 2211.15
Bank Sta=162.9,257.8
XS Rating Curve= 0 ,0
Exp/Cntr(USF)=0,0
Exp/Cntr=0.3,0.1

Type RM Length L Ch R = 1 ,10589   ,369.2,533.1,728.2
XS GIS Cut Line= 2
2231578.05371738443961.2805853452232062.21273423443471.858970478
#Sta/Elev= 30
       0 2193.64    15.7 2193.03    25.8 2195.06    32.7  2194.8    54.2 2184.92
    65.6 2177.38    73.3 2164.49    86.4 2151.13    99.7 2143.57     107 2141.38
   196.4 2141.32   208.3 2141.34   216.5 2143.07   236.2 2147.84   264.6 2147.91
   293.1 2148.24   326.5 2146.16   384.1 2146.07   414.5 2147.37   425.8  2149.3
   445.6 2159.17   452.3 2161.26   496.6 2164.64   530.5 2169.04     539 2169.39
   600.2 2177.33   629.5 2183.72   651.4 2184.94   679.9  2192.3   688.4 2196.45
#Mann= 6 ,-1,0
       0      .1       0    99.7     .04       0   216.5      .1       0
   264.6     .05       0   530.5    .016       0     539     .06       0
#Block Obstruct= 1 ,-1
     472  508.73 2186.12
Bank Sta=99.7,216.5
XS Rating Curve= 0 ,0
Exp/Cntr(USF)=0,0
Exp/Cntr=0.3,0.1

Type RM Length L Ch R = 1 ,10056   ,554.6,645.7,737.5
XS GIS Cut Line= 2
 2231513.4130249443932.1261611042232325.11185584 444574.16311824
#Sta/Elev= 30
       0  2192.5    74.9 2190.85   143.5 2186.12   261.8 2172.55   309.5 2165.35
   330.2 2164.88   364.4 2158.74     386 2152.43   401.4 2149.52   462.5 2141.88
   489.82139.768   508.4 2138.25   580.8 2138.35   588.4 2139.72   605.3 2144.93
     632  2149.9   676.7 2152.67   743.1 2159.53   834.8 2189.94   850.1 2196.59
   865.5 2207.89   879.8 2209.76   906.2 2209.79   911.1 2210.83   923.7 2220.44
     951 2233.37   972.5 2248.22   979.5 2250.11  1023.5  2253.5  1034.9 2258.09
#Mann= 6 ,-1,0
       0      .1       0   489.8     .04       0   588.4      .1       0
   865.5    .016       0   906.2      .1       0   979.5     .06       0
#Block Obstruct= 1 ,-1
  985.52 1010.63 2272.43
Bank Sta=489.8,588.4
XS Rating Curve= 0 ,0
Exp/Cntr(USF)=0,0
Exp/Cntr=0.3,0.1

Type RM Length L Ch R = 1 ,9410    ,527.3,509.5,513.6
Node Name=C
XS GIS Cut Line= 2
2231482.70110669443906.5805297082231256.40939229444601.243466938
#Sta/Elev= 30
       0  2192.7    23.8 2189.29    53.2 2182.68    74.2 2175.27   107.9 2160.75
   120.5 2157.24   137.3 2154.53     150  2153.1   259.4 2146.56   339.3 2148.59
   347.7 2147.29   356.8 2142.91   377.1 2140.74   386.42138.283     394 2136.27
   406.6 2135.51   444.5 2135.41   469.7 2135.46   473.9 2135.88   478.1 2137.84
   486.5 2140.85   494.9 2142.26   503.4 2146.92   543.5 2175.38   575.2 2201.08
   603.8 2218.65   616.5 2220.72     626 2223.46   705.2 2225.81   730.6 2225.37
#Mann= 4 ,-1,0
       0      .1       0   386.4     .04       0   478.1      .1       0
   603.8     .05       0
#Block Obstruct= 1 ,-1
  685.65  712.55 2245.62
Bank Sta=386.4,478.1
XS Rating Curve= 0 ,0
Exp/Cntr(USF)=0,0
Exp/Cntr=0.3,0.1

Type RM Length L Ch R = 1 ,8901    ,601.1,580.8,584.8
XS GIS Cut Line= 2
2231091.48674877443598.578993553  2230781.674689444366.563817784
#Sta/Elev= 30
       0 2174.93    50.6 2167.76   106.3  2157.1   147.8 2152.35   205.5 2149.79
   244.5 2149.13   261.6 2149.93   296.1 2148.83   326.3 2146.27   343.5 2143.06
   360.8 2141.72   382.4 2144.09   403.9 2144.88   532.8 2146.95   539.3 2146.03
   546.3 2141.35   557.52137.424   563.9 2135.82   575.5 2135.01   650.4 2135.16
   654.1  2135.4   659.82137.598   665.3 2140.54   675.7 2142.89   683.8 2146.36
   721.7  2171.5   757.8 2197.77   787.8 2215.82   796.4  2218.3   828.1 2222.61
#Mann= 3 ,0,0
       0      .1       0   557.5     .04       0   659.8      .1       0
Bank Sta=557.5,659.8
XS Rating Curve= 0 ,0
Exp/Cntr(USF)=0,0
Exp/Cntr=0.3,0.1

Type RM Length L Ch R = 1 ,8320    ,204,455,469.9
XS GIS Cut Line= 2
2230668.22238542443192.7688307482230236.23092179444139.659210625
#Sta/Elev= 30
       0 2206.47    35.6 2192.17    57.7 2184.33     106 2172.13   151.3 2163.31
   185.1 2155.48   211.7 2153.17   277.4 2142.31   312.6 2139.97   343.4 2139.34
     361 2140.57   470.9 2142.64   725.9 2146.09   734.7 2145.61   739.1 2143.64
   746.1 2138.39   752.1 2136.99   770.2 2134.79   839.7 2134.68  847.34 2137.04
     871 2141.37   923.7 2143.49   932.5 2145.43   945.4  2146.6   963.3 2156.93
   972.1 2160.71   996.7 2173.59  1005.7 2175.91  1020.5 2175.59  1040.8 2168.98
#Mann= 6 ,-1,0
       0      .1       0   752.1     .04       0  847.34      .1       0
     870     .05       0   996.7      .1       0  1040.8     .03       0
#Block Obstruct= 1 ,-1
 1016.78 1040.78 2195.94
Bank Sta=752.1,847.34
XS Rating Curve= 0 ,0
Exp/Cntr(USF)=0,0
Exp/Cntr=0.3,0.1

Type RM Length L Ch R = 1 ,7865    ,51.7,411.5,438.6
XS GIS Cut Line= 2
2230608.36525516443172.645641239 2229860.9646186443809.843054355
#Sta/Elev= 30
       0 2208.62    37.8 2192.05    68.6 2180.77   136.7 2160.07   163.2 2153.11
   184.2 2145.88   241.3 2140.37   284.4 2138.69   320.9  2140.8   368.2 2140.57
   420.8 2142.37   468.1 2142.54   494.3 2140.75   525.9 2142.96     568 2141.97
     642 2143.39   729.7 2140.92   759.2 2142.83   783.6 2138.12   809.7 2137.77
     827  2134.9   841.82133.854   851.7 2132.44   891.4 2133.39   931.8  2132.6
   942.32134.081   956.9 2142.77   973.7 2161.44   977.9 2165.01   982.2 2166.38
#Mann= 3 ,-1,0
       0      .1       0   841.8     .04       0   942.3      .1       0
Bank Sta=841.8,942.3
XS Rating Curve= 0 ,0
Exp/Cntr(USF)=0,0
Exp/Cntr=0.3,0.1
